HEC-RAS study gum_limited.prj: Gum Swamp

--- gum_limited.g02 (geometry) --- (continued)

Type RM Length L Ch R = 1 ,9119.055,860.68,1133.1,779.41
XS GIS Cut Line= 5
     1842140.526      386783.189     1840742.164       386862.77
     1840344.256       386771.82       1840219.2      386794.558
     1839241.483      386817.295
#Sta/Elev= 30
       0  229.88   48.91  228.07   54.14  221.25   71.65  218.63  106.86  215.73
  108.67   214.4  145.15  211.65  692.03  206.48  810.82  206.35  857.36  204.72
  921.79  200.15  990.79   197.3  996.65   193.1 1064.85   192.6 1335.46  193.88
 1590.71  192.97 1623.59  192.96  1935.9  194.01 1936.72  198.74 1951.71  199.23
 1983.34  202.99  2029.4  205.62 2095.27  206.58 2190.36  205.09 2279.84  207.78
 2475.97  210.44 2641.41  214.75 2757.38  218.87 2848.74   220.3 2913.88  222.42
#Mann= 3 , 0 , 0
       0     .12       0 1590.71    .055       0 1623.59     .12       0
Bank Sta=1590.71,1623.59
Exp/Cntr=.3,.1

Type RM Length L Ch R = 1 ,7985.959,339.1,302.69,253.05
XS GIS Cut Line= 2
     1842129.157      385907.792     1839210.079      386112.116
#Sta/Elev= 30
       0  224.27  112.95  219.95  171.31  219.73  428.19  214.16  459.79  211.94
  560.27   208.5  575.32   206.4  692.71  199.04  810.37  198.17   841.2  196.39
   965.6   195.4 1149.85  195.61 1223.98  196.74 1478.44  195.54 1554.67  196.04
 1605.68  194.71 1611.18  193.62 1644.54  192.64 1644.92  191.81 1677.15  191.65
 2103.81  191.58 2243.14  192.44 2266.88   195.1 2290.77  199.55    2351  204.52
 2391.38  206.67  2475.8   208.8 2699.28  216.96 2750.24  217.68 2926.22   216.9
#Mann= 3 , 0 , 0
       0     .12       0 1644.92    .055       0 1677.15     .12       0
Bank Sta=1644.92,1677.15
Exp/Cntr=.3,.1

Type RM Length L Ch R = 1 ,7683.269,501.34,794.21,684.96
XS GIS Cut Line= 2
     1841805.166      385477.162     1839393.147      385935.141
#Sta/Elev= 30
       0  223.66   44.35  221.72   83.71  220.96   107.7   217.5  120.21  217.38
   129.5   214.9  144.27  214.95  159.36  210.43  215.62  203.05  283.86  197.97
  316.73  197.86  376.26  196.05 1193.22  195.89 1385.02  193.75 1410.46  192.44
 1482.89  191.54  1514.8  191.76 1878.23  190.97 1903.41  191.87 1952.92  192.15
  1970.1  196.27    2004  197.77 2009.29  199.35 2018.57  199.69 2025.38  201.37
 2035.93  202.24  2082.8  204.66 2235.71  208.68  2377.6  215.07 2455.11  214.78
#Mann= 3 , 0 , 0
       0     .12       0 1482.89    .055       0  1514.8     .12       0
Bank Sta=1482.89,1514.8
Exp/Cntr=.3,.1

Type RM Length L Ch R = 1 ,6889.063,354.2,353.13,346.76
XS GIS Cut Line= 2
     1842015.469      385248.402     1838968.632      385032.395
#Sta/Elev= 30
       0   221.4  100.89  220.21  210.22   214.9  289.44  213.73  383.66   208.3
  504.64   198.3  588.95  195.86  671.92   196.8  762.63   195.6  883.64  196.16
 1211.54  193.39 1430.91   194.7 1519.66  194.18  1556.5  193.16 1565.35  192.05
  1637.2  190.38 1667.75  190.66 1832.02   190.2 1952.75  190.34 2093.22  195.09
 2139.31  206.78 2153.74  207.78 2501.45  208.65 2570.37  216.84  2605.1  219.54
 2691.78  220.11 2771.27  227.12 2828.14  229.88 2966.03  231.83 3054.48  232.08
#Mann= 3 , 0 , 0
       0     .12       0  1637.2    .055       0 1667.75     .12       0
Bank Sta=1637.2,1667.75
Exp/Cntr=.3,.1

Type RM Length L Ch R = 1 ,6535.935,560.23,575.49,549.27
XS GIS Cut Line= 2
     1842125.751      384897.057     1839057.296      384698.599
#Sta/Elev= 30
       0  219.23  159.18  218.38  194.84  216.57  474.41  210.31  558.43  206.42
  710.28   202.6  792.07   197.6  922.19  194.65 1303.73  195.38 1452.19  194.34
 1648.48  190.42  1761.9  190.61 1792.65  190.46 1955.11  190.08 2066.34  190.55
 2091.55  195.12 2115.48  196.04 2120.89  197.73 2173.81  202.99 2180.56  204.88
 2192.14  204.58 2238.28  209.03 2526.14  221.78 2620.46  221.74 2666.28  220.13
 2715.88  216.71 2740.29  213.58 2887.06  213.59 2982.23  215.94 3074.87  215.73
#Mann= 3 , 0 , 0
       0     .12       0  1761.9    .055       0 1792.65     .12       0
Bank Sta=1761.9,1792.65
Exp/Cntr=.3,.1

Type RM Length L Ch R = 1 ,5960.443,850.85,942.54,512.8
XS GIS Cut Line= 3
     1842072.313      384316.161       1840217.5      384225.512
     1839225.222      384515.408
#Sta/Elev= 30
       0  209.06  114.98   204.3  259.91  203.58  326.15  202.35  454.34  203.29
  771.49  201.34  862.19  199.85  901.78   196.7  977.36  194.29 1118.56  192.48
 1356.56  192.46 1406.46  191.82 1461.36  189.59 1561.02  189.78 1589.93  189.75
 1836.55  188.85 1975.91  190.34 2006.86  198.32 2023.92  199.69 2044.96  205.42
  2055.3  206.14 2090.24     212 2121.39  215.26 2180.77   215.6 2244.68  214.61
 2293.04  215.79 2440.29  223.34 2558.65  226.08  2741.1  224.49 2890.79  218.89
#Mann= 3 , 0 , 0
       0     .12       0 1561.02    .055       0 1589.93     .12       0
Bank Sta=1561.02,1589.93
Exp/Cntr=.5,.3

Type RM Length L Ch R = 1 ,5017.899,155.01,145.27,168.41
XS GIS Cut Line= 6
     1841857.444      383084.087     1841289.649      383335.674
     1840915.138      383515.418     1840524.971       383682.76
     1840249.348      383791.041     1839562.345      384106.268
#Sta/Elev= 30
    1.88  200.61   30.54  198.22  331.16  198.76  448.89   201.6  584.79  200.31
  649.35  200.69  678.62  194.61   708.6  193.43  869.08   191.9  913.09  192.59
  987.06  190.66 1019.73  189.79 1233.43  190.59 1382.01  188.54 1742.82  189.91
 1795.12  188.51 1917.74  189.45 2003.41  193.32 2043.25  197.22 2062.29  197.43
  2083.3  201.95 2109.67  204.95 2137.14  206.11 2167.11  209.01 2191.49  212.65
 2272.42  221.62 2317.28  224.15  2326.1  225.51 2472.27  233.55 2515.09  234.57
#Mann= 3 , 0 , 0
    1.88     .12       0  987.06    .055       0 1019.73     .12       0
#XS Ineff= 2 , 0
       0   953.4  200.76 1055.77       0  200.76
Bank Sta=987.06,1019.73
Exp/Cntr=.5,.3

Type RM Length L Ch R = 3 ,4945.23 ,,,
BEGIN DESCRIPTION:
Railroad
END DESCRIPTION:
Bridge Culvert--1,0,-1,-1, 0
Deck Dist Width WeirC Skew NumUp NumDn MinLoCord MaxHiCord MaxSubmerge Is_Ogee
60.67,24,2.6,0,120,120,200.76,,.95,0,0,0,,
       0   13.38   18.81   35.34   40.16  189.33  200.59  208.63  214.84  224.48
  249.92  260.94  266.81  279.27   289.4  309.53  325.78  326.36  327.89  449.25
  452.37  464.04  486.97  488.57  593.15  596.05  701.66  711.28  723.93  790.63
  793.42  869.99  889.02  907.57   958.4  1048.4 1162.18 1163.61 1178.77  1264.1
 1269.08 1277.45 1289.35 1294.26 1355.58 1356.86 1371.11 1374.55 1374.87 1390.68
 1391.85 1410.86 1414.54 1434.02 1597.51 1600.79 1614.36 1808.84 1817.85 1856.26
 1861.78 1871.95 1872.82 1873.35 1893.74 1895.76 1970.29 1996.69 1999.47 2017.48
 2018.76 2035.89 2036.37  2036.9 2061.77 2061.94 2062.15 2073.62 2080.63 2084.54
 2093.23 2104.86 2112.24 2142.53 2147.92 2161.55 2164.43 2166.69 2182.49 2184.16
 2186.75 2196.42  2199.7 2210.67 2211.17 2212.43 2232.25 2238.18  2243.7 2251.52
 2264.31 2266.78 2289.25 2293.65 2313.26 2315.05 2315.21 2316.26 2332.44 2336.95
  2352.1 2355.19 2383.33 2384.71 2407.59 2438.72 2472.64 2510.21 2513.05 2513.21
  202.08  201.89   201.8  201.72  201.59     201  200.95  200.95  200.93  201.01
  200.82  200.84  200.88  200.91  200.83  200.85  200.98  200.94  200.95  200.77
   200.8  200.76  200.76   200.8  200.77  200.86  201.57  201.64  201.62  201.61
  201.59  202.21  202.32  202.35   202.9   202.9  203.45  203.55  203.48     204
  204.08  204.22  204.47  204.43   205.1  205.12   205.3  205.29  205.34  205.42
  205.41  205.63  205.64   205.9  207.27  207.26  207.49  208.81   208.8  209.26
  209.55  210.02  210.05  210.07  210.35  210.33  210.78  211.06  211.17  211.68
  211.87  212.05  212.04  212.05   212.2   212.2  212.21  212.51  212.66  212.73
  212.83   213.1  213.14  213.33  213.37  213.77  213.84  213.92  213.97  213.95
  214.05  214.23  214.37   214.5  214.51  214.53   214.6  214.88  215.06  215.44
  215.66  215.75  215.95  215.98  216.37  216.41  216.43   216.4  216.41  216.55
  217.59  217.84  218.04  217.99  218.44  218.62   218.8   218.7  218.73  218.73
                                                                                
                                                                                
                                                                                
                                   200.9   200.9
                                                                                
                                                                                
                                                                                
                                                                                
                                                                                
                                                                                
                                                                                
                                                                                
       0   13.38   18.81   35.34   40.16  189.33  200.59  208.63  214.84  224.48
  249.92  260.94  266.81  279.27   289.4  309.53  325.78  326.36  327.89  449.25
  452.37  464.04  486.97  488.57  593.15  596.05  701.66  711.28  723.93  790.63
  793.42  869.99  889.02  907.57   958.4  1048.4 1162.18 1163.61 1178.77  1264.1
 1269.08 1277.45 1289.35 1294.26 1355.58 1356.86 1371.11 1374.55 1374.87 1390.68
 1391.85 1410.86 1414.54 1434.02 1597.51 1600.79 1614.36 1808.84 1817.85 1856.26
 1861.78 1871.95 1872.82 1873.35 1893.74 1895.76 1970.29 1996.69 1999.47 2017.48
 2018.76 2035.89 2036.37  2036.9 2061.77 2061.94 2062.15 2073.62 2080.63 2084.54
 2093.23 2104.86 2112.24 2142.53 2147.92 2161.55 2164.43 2166.69 2182.49 2184.16
 2186.75 2196.42  2199.7 2210.67 2211.17 2212.43 2232.25 2238.18  2243.7 2251.52
 2264.31 2266.78 2289.25 2293.65 2313.26 2315.05 2315.21 2316.26 2332.44 2336.95
  2352.1 2355.19 2383.33 2384.71 2407.59 2438.72 2472.64 2510.21 2513.05 2513.21
  202.08  201.89   201.8  201.72  201.59     201  200.95  200.95  200.93  201.01
  200.82  200.84  200.88  200.91  200.83  200.85  200.98  200.94  200.95  200.77
   200.8  200.76  200.76   200.8  200.77  200.86  201.57  201.64  201.62  201.61
  201.59  202.21  202.32  202.35   202.9   202.9  203.45  203.55  203.48     204
  204.08  204.22  204.47  204.43   205.1  205.12   205.3  205.29  205.34  205.42
  205.41  205.63  205.64   205.9  207.27  207.26  207.49  208.81   208.8  209.26
  209.55  210.02  210.05  210.07  210.35  210.33  210.78  211.06  211.17  211.68
  211.87  212.05  212.04  212.05   212.2   212.2  212.21  212.51  212.66  212.73
  212.83   213.1  213.14  213.33  213.37  213.77  213.84  213.92  213.97  213.95
  214.05  214.23  214.37   214.5  214.51  214.53   214.6  214.88  215.06  215.44
  215.66  215.75  215.95  215.98  216.37  216.41  216.43   216.4  216.41  216.55
  217.59  217.84  218.04  217.99  218.44  218.62   218.8   218.7  218.73  218.73
                                                                                
                                                                                
                                                                                
                                   200.9   200.9
                                                                                
                                                                                
                                                                                
                                                                                
                                                                                
                                                                                
                                                                                
                                                                                
BR Coef=-1 , 1 , 0 ,, 0 ,,,.8,0,1.2,0,
WSPro=,,,, 1 ,,,, 0 ,,,, 0 ,,,,-1 ,-1 ,-1 , 0 , 0 , 0 , 0 , 0
BC Design=,, 0 ,, 0 ,,,,,,

Type RM Length L Ch R = 1 ,4872.627,209.01,480.58,327.38
XS GIS Cut Line= 6
     1841816.855      382950.325      1841249.06      383201.912
     1840874.548      383381.657     1840484.381      383548.999
     1840208.759      383657.279     1839521.755      383972.506
#Sta/Elev= 30
   -1.88  200.95   99.33  199.29  267.29   199.2  365.08  196.19  518.04  193.32
  803.17  192.18  842.07  191.12  909.95  191.19  985.81  188.52 1020.99  187.79
 1023.86  187.62 1346.77   188.3 1454.62  189.32 1528.28  188.31 1580.19  188.44
 1665.28     190 1735.38  194.17 1771.36  198.28  1826.2  202.41 1977.19  205.73
 2031.23  208.85 2039.16  210.28 2068.09  211.91 2199.37  213.71 2306.07  213.91
 2368.85  217.07 2400.67  219.38 2479.37   227.4 2497.31   228.6 2511.33  230.94
#Mann= 3 , 0 , 0
   -1.88     .12       0  985.81    .055       0 1020.99     .12       0
#XS Ineff= 2 , 0
       0   953.4  200.76 1055.77       0  200.76
Bank Sta=985.81,1020.99
Exp/Cntr=.5,.3

Type RM Length L Ch R = 1 ,4392.048,356.38,355.95,352.7
XS GIS Cut Line= 4
      1841796.01      382892.371     1840362.973      383256.031
     1839879.902      383068.548     1839575.343      383115.291
#Sta/Elev= 30
       0  200.12    47.1  199.07  219.96  198.91   278.8  196.37  325.84  195.34
  394.32  195.93  458.73  198.27  538.44  194.93  728.65  191.66  787.03  191.74
  854.68   193.4  923.29  192.57  948.05   191.3  970.45  188.96  1357.5  188.23
 1380.92  187.99 1387.47  188.08  1417.4  188.59 1468.22  192.02 1479.02  196.38
 1510.32  201.94 1515.78  203.58 1645.77  203.57 1731.91  207.87 1762.36  210.18
 1841.18  212.13 1967.44  217.58 2095.13   220.5 2231.72  224.79 2304.76   225.9
#Mann= 3 , 0 , 0
       0     .12       0  1357.5    .055       0 1387.47     .12       0
Bank Sta=1357.5,1387.47
Exp/Cntr=.3,.1

Type RM Length L Ch R = 1 ,4036.102,277.88,382.29,385.9
XS GIS Cut Line= 3
     1841662.788      382557.516     1840028.117      382982.386
     1839581.643      382982.386
#Sta/Elev= 30
       0  197.37    73.1  196.41   84.71  194.17  162.63  191.34  205.99  191.26
  299.99  192.81  380.05  192.05  530.65   192.4  634.98  191.31  861.14  192.99
   901.1  192.49  922.53  187.84  945.61  187.23 1156.42  187.58 1204.72  186.96
 1291.95  187.69 1323.98  188.38 1388.05  188.38 1451.98  192.84 1470.89  196.45
 1480.98  197.08 1525.18  203.03 1530.76  202.92 1587.12  212.14 1685.75  212.21
  1801.7  217.95 1891.39  218.58 1977.61  220.96 2001.63  222.48 2135.46     226
#Mann= 3 , 0 , 0
       0     .12       0 1291.95    .055       0 1323.98     .12       0
Bank Sta=1291.95,1323.98
Exp/Cntr=.5,.3

Type RM Length L Ch R = 1 ,3653.810,243.77,282.63,250.97
XS GIS Cut Line= 5
     1842061.406      382399.215     1840539.773      382511.729
     1840088.266      382549.808     1839865.233      382587.887
     1839669.399      382653.165
#Sta/Elev= 30
  -40.54  198.37   91.26  196.35  169.58   198.3  219.88  197.96  293.13  198.75
  322.98  196.93  381.15  195.25  438.32   195.6  499.97  192.26  533.88  191.62
   750.6  192.22  902.47  191.44  1060.1  192.45 1139.28  191.29 1278.37  192.22
 1396.26  185.94 1748.67185.9646 1780.33186.0028 1818.41  187.01 1848.26  190.76
 1900.61  192.19 1935.32  197.55 2013.77  200.49 2033.73     203 2094.56  204.02
 2115.03  207.88  2128.9  208.79 2231.35  210.66 2315.16  214.01 2371.05  217.47
#Mann= 3 , 0 , 0
  -40.54     .12       0 1748.67    .055       0 1780.33     .12       0
#XS Ineff= 2 , 0
       0  1714.5  193.22  1814.5       0  193.22
Bank Sta=1748.67,1780.33
Exp/Cntr=.5,.3

Type RM Length L Ch R = 3 ,3562.55 ,,,
BEGIN DESCRIPTION:
US 74 (NCDOT # 22&23)
END DESCRIPTION:
Bridge Culvert--1,0,-1,-1, 0
Deck Dist Width WeirC Skew NumUp NumDn MinLoCord MaxHiCord MaxSubmerge Is_Ogee
30.76,121,2.6,0,179,179,193.22,,.95,0,0,0,,
       0     .59   26.39   31.64   51.08   59.96   77.73   83.62   94.52  107.96
  111.05  127.55  143.88  150.89  158.08  169.03  182.17  185.17  188.02  205.71
  212.35  215.62  220.39  252.07  253.55  262.18   272.8   283.7   288.7   291.2
  295.16  352.59  375.52  376.24  378.12  396.19  401.44  407.65  417.45  430.52
  434.45  444.38  447.69  467.86  475.19  482.07  502.26  506.72  508.22  511.58
  529.04  536.53  548.42  561.72  569.07  588.01  592.17  595.27   607.9  629.87
  631.59  634.39  648.78  665.36  673.68  695.14  695.53  695.69  696.21  854.37
  893.97  895.01  923.05  927.35  1100.1 1103.47 1281.26 1285.61 1290.95 1315.95
 1479.07 1485.84 1530.57 1531.49 1532.73 1559.57 1560.93 1561.68  1562.3 1593.79
 1594.74 1597.66 1683.58  1686.2 1694.47 1702.05 1705.83  1719.5 1723.73 1723.98
 1729.26 1732.21 1732.54  1809.5 1866.76 1868.32 1883.87  1884.3 1884.33 1896.52
 1899.57  1915.3 1917.28 1920.27 1945.76  1961.8 1963.01  1964.6 1977.55  1984.6
 1987.14 1998.02    2002 2003.42 2013.01 2018.09 2029.72 2034.58 2042.06 2048.86
  2062.2  2070.5 2075.38 2089.86 2094.45 2099.77 2106.38 2115.97 2122.77 2126.68
 2132.96 2139.77 2147.14 2153.79 2160.18 2164.86 2177.74 2188.45 2189.83 2191.41
 2210.87 2215.84 2231.82 2232.69 2233.61 2257.74 2257.95 2258.33 2268.73  2289.1
 2289.29 2302.68 2304.27 2322.11 2323.88 2326.88 2343.25 2343.99 2355.55 2360.15
 2369.11 2369.43 2383.68  2385.9 2397.36 2407.81 2408.87  2410.5 2417.29
  195.88  195.89   195.5  195.45  195.28  195.31  194.93   194.9  194.85  194.84
  194.92  195.28  195.35  195.43  195.31  195.26  194.93  194.89  194.88  194.89
   194.8  194.76  194.79  194.72  194.71  194.67  194.83  194.78  194.84   194.9
  194.86  194.74  194.55  194.56  194.56   194.6  194.65  194.72  194.82  194.81
  194.83  194.96  194.96  194.88  194.78  194.67  194.38  194.32  194.33  194.36
  194.42  194.44  194.32  194.19  194.23  194.22  194.19  194.19  194.31  194.05
  194.04  194.03  194.03  194.11   194.1  193.86  193.86  193.86  193.85  193.83
  193.59  193.62  193.69  193.62  193.27  193.22  193.47  193.54  193.53  193.53
  193.74  193.87  193.98  194.01  194.06  194.15  194.18  194.18  194.15   194.3
  194.29  194.28  194.68  194.62  194.53  194.63  194.69  194.68  194.67  194.66
  194.65  194.65  194.56  195.17  195.77  195.86  195.86  195.86  195.86  195.96
  196.07  196.44  196.48  196.52  197.06  197.27   197.3  197.35  197.86  197.97
  198.01  198.19  198.48  198.52  198.52  198.61  198.96  199.21  199.54  199.77
  200.26  200.57  200.69  201.18  201.26  201.54  201.55  201.75  201.91  202.16
  202.53   202.8     203  203.17   203.2  203.22  203.37  204.15  204.21  204.26
  204.59  204.68  205.15  205.18  205.23  206.79   206.8  206.81  206.88  207.62
  207.62  208.14  208.21  208.74  208.79  208.93  209.57  209.58  210.05  210.24
  210.92  210.94  211.27  211.33  211.47  212.06  212.12  212.19  212.46
                                                                                
                                                                                
                                                                                
                                                                                
                                                                                
                                                                                
                                                                                
                                                                                
                                                                                
                                                          192.65  192.65  192.65
  192.65  192.65  192.65  192.65
                                                                                
                                                                                
                                                                                
                                                                                
                                                                                
                                                                                
                                                                        
       0     .59   26.39   31.64   51.08   59.96   77.73   83.62   94.52  107.96
  111.05  127.55  143.88  150.89  158.08  169.03  182.17  185.17  188.02  205.71
  212.35  215.62  220.39  252.07  253.55  262.18   272.8   283.7   288.7   291.2
  295.16  352.59  375.52  376.24  378.12  396.19  401.44  407.65  417.45  430.52
  434.45  444.38  447.69  467.86  475.19  482.07  502.26  506.72  508.22  511.58
  529.04  536.53  548.42  561.72  569.07  588.01  592.17  595.27   607.9  629.87
  631.59  634.39  648.78  665.36  673.68  695.14  695.53  695.69  696.21  854.37
  893.97  895.01  923.05  927.35  1100.1 1103.47 1281.26 1285.61 1290.95 1315.95
 1479.07 1485.84 1530.57 1531.49 1532.73 1559.57 1560.93 1561.68  1562.3 1593.79
 1594.74 1597.66 1683.58  1686.2 1694.47 1702.05 1705.83  1719.5 1723.73 1723.98
 1729.26 1732.21 1732.54  1809.5 1866.76 1868.32 1883.87  1884.3 1884.33 1896.52
 1899.57  1915.3 1917.28 1920.27 1945.76  1961.8 1963.01  1964.6 1977.55  1984.6
 1987.14 1998.02    2002 2003.42 2013.01 2018.09 2029.72 2034.58 2042.06 2048.86
  2062.2  2070.5 2075.38 2089.86 2094.45 2099.77 2106.38 2115.97 2122.77 2126.68
 2132.96 2139.77 2147.14 2153.79 2160.18 2164.86 2177.74 2188.45 2189.83 2191.41
 2210.87 2215.84 2231.82 2232.69 2233.61 2257.74 2257.95 2258.33 2268.73  2289.1
 2289.29 2302.68 2304.27 2322.11 2323.88 2326.88 2343.25 2343.99 2355.55 2360.15
 2369.11 2369.43 2383.68  2385.9 2397.36 2407.81 2408.87  2410.5 2417.29
  195.88  195.89   195.5  195.45  195.28  195.31  194.93   194.9  194.85  194.84
  194.92  195.28  195.35  195.43  195.31  195.26  194.93  194.89  194.88  194.89
   194.8  194.76  194.79  194.72  194.71  194.67  194.83  194.78  194.84   194.9
  194.86  194.74  194.55  194.56  194.56   194.6  194.65  194.72  194.82  194.81
  194.83  194.96  194.96  194.88  194.78  194.67  194.38  194.32  194.33  194.36
  194.42  194.44  194.32  194.19  194.23  194.22  194.19  194.19  194.31  194.05
  194.04  194.03  194.03  194.11   194.1  193.86  193.86  193.86  193.85  193.83
  193.59  193.62  193.69  193.62  193.27  193.22  193.47  193.54  193.53  193.53
  193.74  193.87  193.98  194.01  194.06  194.15  194.18  194.18  194.15   194.3
  194.29  194.28  194.68  194.62  194.53  194.63  194.69  194.68  194.67  194.66
  194.65  194.65  194.56  195.17  195.77  195.86  195.86  195.86  195.86  195.96
  196.07  196.44  196.48  196.52  197.06  197.27   197.3  197.35  197.86  197.97
  198.01  198.19  198.48  198.52  198.52  198.61  198.96  199.21  199.54  199.77
  200.26  200.57  200.69  201.18  201.26  201.54  201.55  201.75  201.91  202.16
  202.53   202.8     203  203.17   203.2  203.22  203.37  204.15  204.21  204.26
  204.59  204.68  205.15  205.18  205.23  206.79   206.8  206.81  206.88  207.62
  207.62  208.14  208.21  208.74  208.79  208.93  209.57  209.58  210.05  210.24
  210.92  210.94  211.27  211.33  211.47  212.06  212.12  212.19  212.46
                                                                                
                                                                                
                                                                                
                                                                                
                                                                                
                                                                                
                                                                                
                                                                                
                                                                                
                                                          192.65  192.65  192.65
  192.65  192.65  192.65  192.65
                                                                                
                                                                                
                                                                                
                                                                                
                                                                                
                                                                                
                                                                        
BR Coef=-1 , 1 , 0 ,, 0 ,,,.8,0,1.2,0,
WSPro=,,,, 1 ,,,, 0 ,,,, 0 ,,,,-1 ,-1 ,-1 , 0 , 0 , 0 , 0 , 0
BC Design=,, 0 ,, 0 ,,,,,,

Type RM Length L Ch R = 1 ,3371.178,296.18,662.32,619.58
XS GIS Cut Line= 5
     1842061.406      382157.803     1840534.081      382270.738
     1840082.574      382308.817      1839859.54      382346.895
     1839663.706      382412.174
#Sta/Elev= 30
   40.54  197.03  100.78  197.54  150.37  196.46  179.66  196.77  222.32  195.59
  281.95   195.9  308.29  195.35  388.53  197.04  418.07  198.35  482.72  199.12
   559.8  195.73  644.35  189.05  714.67  187.77   959.5  185.99 1396.26  185.94
 1746.27  185.97  1782.7  186.01 1808.46  186.38 1825.87  187.72 1848.26  190.76
 1880.27  196.97 1967.43  204.02 1989.75  207.73 2016.61  208.14  2030.6  207.32
 2111.47  206.43  2202.6  206.36 2304.02  208.89 2405.34  212.65 2457.83   213.7
#Mann= 3 , 0 , 0
   40.54     .12       0 1746.27    .055       0  1782.7     .12       0
#XS Ineff= 2 , 0
       0  1714.5  192.65  1814.5       0  192.65
Bank Sta=1746.27,1782.7
Exp/Cntr=.5,.3

Type RM Length L Ch R = 1 ,2708.859,378.78,472.05,394.36
XS GIS Cut Line= 4
     1841627.489      382134.232     1841393.576      382155.991
     1840906.499      381946.038     1839646.574      381402.664
#Sta/Elev= 30
       0  197.28   76.11  194.77  160.89  189.38  187.97  188.62  311.49  187.74
   354.8  185.89  428.78  186.18  558.14  185.54   876.6  187.34  982.34  187.34
 1000.17  185.59 1015.94  187.36 1062.74   187.7 1092.96  191.91 1100.45  191.91
 1115.62   194.5 1142.31   197.4 1180.23  200.16 1213.24  201.71 1248.24  204.52
 1286.63  205.31 1395.73  203.96 1430.97  204.91 1608.12  204.95 1663.88  203.37
 1731.49  202.63 1781.98   205.1 1873.06  207.83  2064.2  218.74 2137.43  221.38
#Mann= 3 , 0 , 0
       0     .12       0  982.34    .055       0 1015.94     .12       0
Bank Sta=982.34,1015.94
Exp/Cntr=.3,.1

Type RM Length L Ch R = 1 ,2236.808,588.49,829.15,587.99
XS GIS Cut Line= 3
     1841671.007      381796.961     1841371.816      381748.003
     1839808.116      381013.416
#Sta/Elev= 30
       0  196.45   21.59  196.22    94.3  191.71  306.51     192  355.17  190.07
  360.32  189.63   362.9  188.41  442.99  186.19  500.26  185.63  582.05  186.35
   836.7  186.38  850.91   186.1 1097.46  187.28 1260.75  192.86 1273.61  195.19
 1316.02  195.87 1339.14  198.03 1357.78  198.23 1372.27  199.15 1431.59  199.08
 1461.02  199.89 1519.72  199.32 1562.98  199.87 1723.73   203.4 1755.92  204.86
  1803.2  205.73 1881.98  209.27  1923.8  212.97 1943.86  215.64 2030.82  220.91
#Mann= 3 , 0 , 0
       0     .12       0   836.7    .055       0  850.91     .12       0
Bank Sta=836.7,850.91
Exp/Cntr=.3,.1

Type RM Length L Ch R = 1 ,1407.654,442.54,629.71,412.68
XS GIS Cut Line= 4
     1841987.557      381468.773     1841583.455      381235.218
     1841037.753      380985.104     1840153.292      380583.877
#Sta/Elev= 30
       0  194.16   49.62  194.72   56.68  193.48   87.86  193.14  109.55  191.85
  178.54  190.43  373.02  188.43  422.43  185.79  561.19  185.36  618.42   185.8
  717.46  185.59  748.03  185.75   830.5  185.57   836.4  187.98  892.45  190.24
  921.88  190.52 1028.42  194.59 1145.85  197.17 1189.39  200.35 1233.86   204.7
 1255.86  205.25 1303.38  205.72 1450.61  202.94 1623.19  202.49 1851.34  206.99
 1907.88  208.53  1920.3  208.38 1958.46  211.23 1994.46  212.95 2038.24  214.25
#Mann= 3 , 0 , 0
       0     .12       0  717.46    .055       0  748.03     .12       0
Bank Sta=717.46,748.03
Exp/Cntr=.3,.1

Type RM Length L Ch R = 1 ,777.945 ,329.17,499.82,329.92
XS GIS Cut Line= 4
     1842699.137      381318.255     1841888.601      380959.226
     1841540.451      380779.711     1840245.769      380192.208
#Sta/Elev= 30
       0  198.95  303.71  196.89  378.33  193.92  512.85   190.5   575.1  188.39
  610.67  186.33   616.6  185.22   997.8  185.08 1014.73  184.73 1033.07   185.1
 1560.98  185.09 1601.07  191.51 1643.07  192.84 1664.96  196.81  1753.9  198.57
 1791.47  198.88 1852.11  201.32 1917.57  203.11 2009.52  203.26 2081.74  201.63
 2131.91  201.27 2252.47  202.37 2342.51  203.84 2427.89  205.94 2500.16  206.75
 2525.85  208.08 2554.75  208.64 2597.98  210.65 2667.42  214.83 2699.95  216.28
#Mann= 3 , 0 , 0
       0     .12       0   997.8    .055       0 1033.07     .12       0
Bank Sta=997.8,1033.07
Exp/Cntr=.3,.1

Type RM Length L Ch R = 1 ,278.122 ,238.2,277.84,233.66
XS GIS Cut Line= 5
     1842743.396      381007.045     1842038.207      380666.778
     1841617.561       380462.14     1841526.611      380450.771
      1840373.36      379952.567
#Sta/Elev= 30
       0  200.46  126.56  199.53  235.81  196.13  298.52  196.09  380.86  194.56
  415.95  191.95  425.64  190.27  439.31  189.46  567.41  188.09 1017.91   187.3
 1029.85   184.7 1049.87  187.34  1223.9  187.42 1407.02   188.7 1421.26  190.86
 1447.51  192.42 1460.62  193.87 1495.04  194.71 1527.89  196.55 1600.21   197.5
 1723.28  196.97 1866.49  200.35 1921.04  200.84 1985.26  200.23 2075.04  201.43
 2183.17   204.2 2355.34  210.29 2407.47  210.91  2458.1  212.73 2598.69  215.75
#Mann= 3 , 0 , 0
       0     .12       0 1017.91    .055       0 1049.87     .12       0
Bank Sta=1017.91,1049.87
Exp/Cntr=.3,.1

Type RM Length L Ch R = 1 ,0.282   ,.58,.28,.58
XS GIS Cut Line= 3
     1842825.153      380724.961     1841292.869      380124.066
     1840523.934      379789.861
#Sta/Elev= 30
       0  200.55  217.33   198.1  333.67  198.63  445.73  193.87  470.98  191.49
  592.04  187.38   679.1   185.6  848.36  184.89  866.78  184.74  882.43  184.87
 1093.14  184.89  1112.7   185.5 1146.61  187.73 1150.59  189.01 1163.02  190.05
 1231.85  190.17    1358  196.65 1449.08  196.73 1594.82  195.76 1712.11  197.76
 1817.55  198.46  1875.1  200.13 1956.21  200.86 2033.17  203.39 2118.66  204.34
 2249.05  208.17 2295.81  208.96 2403.68  213.38 2449.27  213.76 2484.32  215.53
#Mann= 3 , 0 , 0
       0     .12       0  848.36    .055       0  882.43     .12       0
Bank Sta=848.36,882.43
Exp/Cntr=.3,.1

Chan Stop Cuts=-1

--- gum_limited.g01 (geometry) ---

Geom Title=Base Geometry
Version=September 1998 Version 2.2

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
River Reach=Gum Swamp       ,Reach 01

Type RM Length L Ch R = 1 ,56146.35,381.51,430.88,359.51
XS GIS Cut Line= 2
     1832251.916      417047.607     1831124.716      416612.098
#Sta/Elev= 30
       0  257.23   11.06  257.39   57.93  256.25   73.39  254.63  122.84  252.79
  142.26  252.55  202.24  249.89  269.11  244.96  290.91  241.99  310.17  241.22
  313.49  239.93  366.81  236.68  379.56  236.51   402.4  237.27  432.61  237.02
  485.24  236.55  560.33  238.17  738.83  239.72  779.88  242.55  804.62  242.47
  853.73  246.09  863.79  247.81  888.45  248.89  945.84  259.42 1025.02  269.34
 1057.95  271.41 1071.22  272.76 1117.07  274.57 1139.43  274.75 1208.41  273.55
#Mann= 0 , 0 , 0
Bank Sta=402.4,432.61
Exp/Cntr=.3,.1

Type RM Length L Ch R = 1 ,55715.47,602.68,802.38,587.97
XS GIS Cut Line= 2
     1832568.731      416844.907      1831147.04      416200.515
#Sta/Elev= 30
       0  256.61   51.15   256.8   70.11  256.37  150.23  251.61  179.43  247.48
  201.04   245.1  252.41  243.68  281.79  237.79  448.83  236.02   538.2  236.37
  552.51  235.98  568.17  236.37   607.1  236.31  702.24  238.74   764.6  239.51
  789.93  240.71   843.8  240.06  861.91  240.37  959.48  245.42 1004.04   249.8
 1053.17  250.06 1078.79  252.25 1174.56  254.13 1232.49  261.57  1287.8   267.7
 1310.48  271.13 1333.87  272.68 1350.85  274.88 1426.44  280.81 1560.91  289.52
#Mann= 0 , 0 , 0
Bank Sta=538.2,568.17
Exp/Cntr=.3,.1

Type RM Length L Ch R = 1 ,54913.09,403.79,499.25,384.19
XS GIS Cut Line= 2
     1833229.233      416514.656      1831545.62      415756.051
#Sta/Elev= 30
       0  254.06  117.33  255.23  220.28  254.24  340.27  247.88  395.88  244.08
  450.86  241.95   475.2  238.83  531.82  238.54  628.86  236.87  676.39  237.01
  826.62  235.99  893.64  236.36  909.01  235.43  925.16  235.51  1009.6  236.75
  1151.6  246.65 1157.48  246.48 1176.73  247.95 1215.82  253.48 1261.63  258.48
 1308.54  265.25  1366.8   272.3 1442.43  278.64  1464.3   279.9 1493.07  281.14
 1598.18  283.89 1645.94   284.1 1725.28  285.62 1775.51  285.77 1846.63  284.62
#Mann= 0 , 0 , 0
Bank Sta=893.64,925.16
Exp/Cntr=.3,.1

Type RM Length L Ch R = 1 ,54413.84,649.56,884.73,623.49
XS GIS Cut Line= 2
     1833266.829      416110.024     1831778.827      415442.434
#Sta/Elev= 30
       0  253.74   45.15  252.31   63.09  249.52  112.56  246.79  134.72  244.59
  160.17  244.33  170.27  242.57  435.97  241.96  505.33     240  554.15  237.07
  665.77  237.56  680.68  236.54  688.72  235.05  707.33  234.98  797.51  235.11
  826.86  235.08  922.11  236.05  978.04  238.57 1010.36  244.95 1034.78  245.56
 1069.71  250.71 1088.29  251.85  1146.2     258 1206.66  266.31 1311.19  274.61
 1331.38  277.29 1402.43  280.74 1439.93   280.6 1481.77  281.83  1630.9  290.82
#Mann= 0 , 0 , 0
Bank Sta=797.51,826.86
Exp/Cntr=.3,.1

Type RM Length L Ch R = 1 ,53529.10,701.43,950.8,678.49
XS GIS Cut Line= 3
     1833664.198      415648.754     1832367.358      415056.719
     1832194.178      414698.276
#Sta/Elev= 30
       0  254.12  279.39  253.13  355.22  249.88  369.91  246.28  378.23  246.37
  387.84  244.59  403.72  244.41  416.79   242.1  476.16  239.04  511.98  237.82
  557.24  237.76  584.87  236.27  643.49  236.49  767.77  234.88  788.59  234.86
  795.12  234.93  945.76  236.26   985.1  240.79 1016.64  245.55 1073.78  246.73
 1133.13   250.4 1241.68  263.45 1258.57  266.53 1272.91  267.91 1298.14  271.94
 1357.35  277.39 1442.37  280.88 1627.63  282.96 1710.11  286.66 1823.67  293.07
#Mann= 0 , 0 , 0
Bank Sta=767.77,795.12
Exp/Cntr=.3,.1

Type RM Length L Ch R = 1 ,52578.30,757.77,773.92,737.85
XS GIS Cut Line= 2
     1834063.065      415008.227     1832365.938      414404.983
#Sta/Elev= 30
       0  254.28   62.47  254.62  326.03  249.09  363.03  250.28  482.56  250.06
  525.55  248.38  573.28  244.47  595.46  243.64  620.09  240.36  634.03  237.31
  659.58  235.48  690.31  234.65  847.15  234.89  915.21  233.88  947.68  233.87
 1143.66  236.94 1161.92  238.44 1179.52  241.41 1195.95  246.46 1265.68     248
 1308.59   255.8 1366.27  261.97 1438.04  273.74 1480.55  275.42 1525.86  275.64
 1587.61  278.07 1712.32  288.41 1725.73  290.19 1747.09  290.78 1801.15  294.72
#Mann= 0 , 0 , 0
Bank Sta=915.21,947.68
Exp/Cntr=.5,.3

Type RM Length L Ch R = 1 ,51804.38,144.8,147.06,148.22
XS GIS Cut Line= 6
     1834365.974      414345.483     1834164.601      414220.632
     1833105.381      413898.436     1832940.256      413817.887
     1832795.268      413721.228     1832428.769      413358.757
#Sta/Elev= 30
   -3.31  246.71   76.41   240.8  160.85  238.93  286.03  241.35   328.2  240.74
  371.99  241.57  506.16   239.6  572.53  239.95  646.99  238.02  908.23  239.07
  972.61  233.64 1096.34  233.15 1112.28  233.03 1127.88   233.2 1148.69  235.83
 1220.92  240.05 1254.57  241.12 1272.13  242.92 1298.92  243.39 1328.67  245.86
 1371.96  247.52 1414.96  251.53 1482.28  253.84 1528.11  254.27 1700.93  260.69
 1796.82  271.48  1857.5   274.6 1932.27  274.05 2074.94  279.43  2214.3  281.68
#Mann= 3 , 0 , 0
   -3.31               0 1096.34               0 1127.88               0
#XS Ineff= 2 , 0
          904.65  239.11
Bank Sta=1096.34,1127.88
Exp/Cntr=.5,.3

Type RM Length L Ch R = 1 ,51657.32,276.96,425.37,285.74
XS GIS Cut Line= 6
     1834432.738      414217.089     1834231.366      414092.238
     1833172.146      413770.042      1833007.02      413689.493
     1832862.032      413592.834     1832495.534      413230.364
#Sta/Elev= 30
    3.31  242.96  112.28  245.07  263.15  241.53  508.31  240.26  640.14  238.95
  672.64  237.65  722.02  237.17  869.84  237.21  942.26  235.99  968.93  234.45
 1096.37  233.59 1112.93  233.49 1127.79   233.6 1135.94  235.31 1164.87  237.66
 1226.24  240.81 1322.77  243.78 1432.95  249.16 1468.58  254.09 1481.39  255.01
 1520.07  255.17 1544.05  256.31 1741.16  267.26 1767.21  269.36 1908.81  276.03
 1961.99  279.73 2015.64  281.88 2025.99  283.32 2113.59  290.01 2220.91  295.48
#Mann= 3 , 0 , 0
    3.31               0 1096.37               0 1127.79               0
Bank Sta=1096.37,1127.79
Exp/Cntr=.5,.3

Type RM Length L Ch R = 1 ,51231.95,328.89,345.87,386.51
XS GIS Cut Line= 4
     1834360.947      414158.597     1833684.335      413651.138
     1833168.821      413457.821     1832778.158       413063.13
#Sta/Elev= 30
       0  245.19   27.12  245.28  112.37  242.28  261.46     239  340.26  238.77
  385.67  236.62  811.02  240.27  845.76  238.07  870.41   234.8   927.7  232.79
  952.41  232.93  991.45  233.79  1056.2  234.47 1147.47  238.36 1202.36  238.63
 1219.44  241.21 1259.04  241.63  1374.9  255.27 1395.59  255.61 1425.51  259.24
 1464.54  262.23 1489.11   265.7 1513.16  266.42 1563.45  271.38 1659.45  276.53
 1812.34  291.35 1838.81  295.83 1867.26  299.14 1924.88  303.45 1951.67  304.01
#Mann= 0 , 0 , 0
Bank Sta=952.41,991.45
Exp/Cntr=.3,.1

Type RM Length L Ch R = 1 ,50886.07,408.69,544.35,585.92
XS GIS Cut Line= 3
     1834352.892      414130.405     1833406.441      412825.511
     1833305.754      412483.177
#Sta/Elev= 30
       0  245.39   28.23  244.95    94.7  242.54  132.51  238.69  144.19  239.18
  163.43  237.93  257.51  235.58  370.98  235.29  419.28  234.12  479.11  234.54
  559.46  231.82  708.81  231.49     811  233.62  943.07  232.82  958.07  231.32
  972.92  232.79 1070.76  233.73 1120.35  238.15 1180.77  237.48 1238.23  237.78
 1287.61   241.6 1312.86  241.82 1365.58  247.52 1444.37  252.94 1486.95  254.51
 1528.34  258.52  1598.7  261.95 1616.64  264.14  1701.4  271.38 1968.83   291.8
#Mann= 0 , 0 , 0
Bank Sta=943.07,972.92
Exp/Cntr=.3,.1

Type RM Length L Ch R = 1 ,50341.72,960.52,887.71,761.47
XS GIS Cut Line= 4
     1834904.653      414303.585     1834360.947      414110.268
     1834330.256      413910.691     1834244.084      412715.771
#Sta/Elev= 30
       0  239.35   10.82  238.32   30.54  237.98  176.68  239.34  234.91  241.01
   291.3  241.57  410.93  240.37   515.2  241.75  577.05  245.48  600.24  244.97
  673.94  237.48  690.61  237.03  725.81  234.13 1079.94     233 1201.28  233.39
 1226.86  233.15 1247.48  231.56 1259.43  231.41 1279.31  231.55 1313.17  233.08
 1394.05  233.77 1439.97  235.32 1485.79  239.47 1517.33  241.14  1570.8  243.71
 1658.95  246.43 1780.98  254.99 1835.55   257.2 1933.84  258.61    1977  260.38
#Mann= 0 , 0 , 0
Bank Sta=1247.48,1279.31
Exp/Cntr=.3,.1

Type RM Length L Ch R = 1 ,49454.01,417.49,432.71,448.53
XS GIS Cut Line= 2
     1835555.135      413761.394     1834493.425      412659.469
#Sta/Elev= 30
       0   245.6   22.21  244.56   63.79  244.27  128.53  241.81  167.97  241.49
  214.09   239.2     255  233.43  276.16  232.23  339.36  230.47  575.55  229.17
  638.62  229.83  711.54  228.97  742.25  228.83  771.96  233.02  855.47  236.65
  875.84  236.85  935.34  235.42     964  235.64 1042.28  238.66  1149.2  239.35
 1189.09  241.08 1271.44  240.96 1350.72  242.88 1376.89  245.99 1399.45  246.68
 1426.53  251.51 1450.03  253.95 1472.04  258.71 1495.21  261.25 1530.19   266.4
#Mann= 0 , 0 , 0
Bank Sta=711.54,742.25
Exp/Cntr=.3,.1

Type RM Length L Ch R = 1 ,49021.30,448.7,507.06,494.18
XS GIS Cut Line= 2
     1835909.038      413568.356     1834887.545      412410.128
#Sta/Elev= 30
       0  247.52   23.45  247.12   61.88  245.19  106.26  243.64   170.5  242.55
  215.96   242.3  345.33   239.7  391.16  236.91  396.84  235.59  512.32  229.52
  744.03  228.79  807.54  228.95  838.57  229.55     969  229.91 1015.11  230.95
 1049.06  230.93 1112.91  231.78 1138.29  232.97 1156.95  234.38 1182.71  234.75
 1197.92  235.56 1250.64  236.87 1267.77  238.57 1292.64  238.66 1331.77  240.96
 1348.81  241.03 1357.04  241.79 1392.46  243.31 1449.19  246.78 1544.32   250.8
#Mann= 0 , 0 , 0
Bank Sta=807.54,838.57
Exp/Cntr=.3,.1

Type RM Length L Ch R = 1 ,48514.24,491.98,530.75,498.95
XS GIS Cut Line= 4
     1836421.645      413438.861     1835943.735      412970.499
     1835476.551      412265.695     1835347.672      412104.597
#Sta/Elev= 30
       0  245.63   37.75  243.15     123  240.06  195.27  239.45  452.61  240.59
  554.56  239.31  627.98  236.54  672.35   236.4  694.57  230.41  736.27  230.83
  809.56  228.58  930.33  228.46  980.34  228.93 1007.55  230.15 1034.48  230.08
 1049.55  228.42  1070.4  230.08 1112.12  231.73 1189.94   232.1 1260.45  234.07
 1350.39  234.55 1406.75  236.95 1435.87   238.7 1470.35   241.7 1479.12  243.45
 1501.31  244.55 1585.26  254.01 1643.39  257.71 1658.64  260.33 1721.04  265.13
#Mann= 0 , 0 , 0
Bank Sta=1034.48,1070.4
Exp/Cntr=.3,.1

Type RM Length L Ch R = 1 ,47983.48,604.09,833.02,405.68
XS GIS Cut Line= 3
     1836684.786      413328.942     1836507.578      412962.444
     1835770.555      411842.813
#Sta/Elev= 30
       0  251.97   59.91   249.2   95.82  248.67  210.02  243.19  272.82  242.94
  299.31  241.61  393.24  240.57  418.48  239.11  486.39  237.63  514.27  234.13
  557.17  234.03   585.2  231.34   747.2  227.73  864.53  228.19  997.84  230.13
 1011.94  227.98 1031.04  231.61 1050.63  231.53 1102.38  234.99 1156.67  234.47
 1172.81   233.6 1216.73  234.12 1266.22  233.57 1483.04  236.75 1520.99  239.67
 1575.59  242.11 1599.78  244.46 1671.74   253.2  1688.1  256.16 1747.53   262.8
#Mann= 0 , 0 , 0
Bank Sta=997.84,1031.04
Exp/Cntr=.3,.1

Type RM Length L Ch R = 1 ,47150.46,418.16,702.26,775.76
XS GIS Cut Line= 3
     1836809.637      413304.777     1836781.445       412241.53
      1835984.01      411738.099
#Sta/Elev= 30
       0  249.22  114.67  245.68  242.82  240.26  310.39   240.3  352.96  242.96
  387.57  242.82  440.06  241.08  457.63  239.02  509.66  235.41  527.35  235.06
  617.02  234.21  670.36  234.51   682.9  235.64  701.54   235.8  865.79  233.39
 1113.98  233.93 1186.47  230.57 1226.89  230.41 1252.98     228 1274.24  227.38
 1303.12  227.07 1304.34  227.15 1402.06  228.63 1423.55  230.95 1557.17  231.03
 1709.46  233.05 1780.28  238.21    1827   239.9 1918.51  249.57 2006.67  256.42
#Mann= 0 , 0 , 0
Bank Sta=1274.24,1304.34
Exp/Cntr=.5,.3

Type RM Length L Ch R = 1 ,46448.20,219.62,230.38,192.73
XS GIS Cut Line= 6
     1836927.342      413178.914     1836917.594       412678.25
     1836798.464      412099.557     1836891.095      411672.648
     1836911.232      411459.193      1836677.64      410915.487
#Sta/Elev= 30
   36.77  245.81   87.64   245.1  199.89  241.03  252.63  241.26  330.49  243.99
  367.26  243.82  425.35  240.88  590.36  236.99  697.97  239.28  865.25  234.05
 1071.33  234.15 1239.83  231.85  1302.2  229.62 1403.77  228.95 1452.62  227.06
  1542.6  227.57 1577.62   226.9 1633.79  226.37 1754.25  226.79 1869.31  230.49
 1929.44  234.88 1963.11  239.23 2057.02  246.65 2077.79  250.29 2115.55   251.2
  2136.5  256.84 2174.99  257.24 2208.41   262.3 2300.68  269.31 2371.39  271.49
#Mann= 3 , 0 , 0
   36.77               0  1542.6               0 1577.62               0
Bank Sta=1542.6,1577.62
Exp/Cntr=.5,.3

Type RM Length L Ch R = 1 ,46217.82,221.29,193.51,178.78
XS GIS Cut Line= 6
     1837118.842      413173.875     1837109.094      412673.211
     1836989.964      412094.518     1837082.595      411667.608
     1837102.732      411454.153      1836869.14      410910.447
#Sta/Elev= 30
  -36.77  247.78   18.44  244.58   84.28   243.9  119.17  242.76  286.51   242.3
  362.77  243.53  450.99  241.57  572.38  241.88  617.09  241.25   836.2  233.44
 1176.68  226.46 1393.83  227.12 1536.76  226.34 1549.21  226.03 1583.46  226.72
  1614.5  226.68 1664.57  230.08 1771.06  230.61 1785.45  237.52 1812.02  238.98
  1826.6  242.29  1834.7  245.38 1841.76  246.63  1905.8  254.83 2008.84  261.58
 2044.34  265.41 2074.15  267.54 2151.26  268.61  2234.7  267.71 2297.85  268.61
#Mann= 3 , 0 , 0
  -36.77               0 1536.76               0 1583.46               0
Bank Sta=1536.76,1583.46
Exp/Cntr=.5,.3

Type RM Length L Ch R = 1 ,46024.32,1016.97,1005.4,786.15
XS GIS Cut Line= 4
     1837409.728      412740.934      1837216.41      412338.189
     1837280.849      411291.052     1837147.943      411081.624
#Sta/Elev= 30
       0  248.52   47.14  247.93   73.68  246.59   83.31  247.63  108.75  246.83
  166.45  246.96  212.43   245.1  260.94  245.14  336.96  246.56  395.75  245.26
  434.44  242.74  453.83  237.02   473.1  233.44  510.89  230.24 1058.48  226.17
 1153.72  226.62 1187.59  225.52 1209.47  225.48 1217.43   225.5 1223.28  230.04
 1232.03  230.83 1337.73  231.27 1377.51  234.08 1420.17  234.41 1481.72  237.63
 1495.99  238.91 1584.37  256.09 1603.52  257.45 1622.23  260.05  1743.9  267.71
#Mann= 0 , 0 , 0
Bank Sta=1187.59,1217.43
Exp/Cntr=.3,.1

Type RM Length L Ch R = 1 ,45018.92,517.35,928.06,885.9
XS GIS Cut Line= 3
     1838307.849      412571.781     1838195.081      411713.934
      1837832.61      410783.593
#Sta/Elev= 30
       0  249.47   68.42   245.8  191.32  244.04  316.28  245.58  417.45  240.21
  510.98  240.46  607.48  237.47  642.46  237.25  711.47  233.45  740.07  230.43
   795.9  229.29  812.82  228.19  817.25  227.09  836.69  226.54  897.69  225.27
 1190.14  224.54 1308.04  225.86 1325.37  224.69  1347.9  225.87 1466.67  227.45
 1566.62  232.31 1583.65  237.57 1590.44  238.35 1678.38  240.97 1710.82  244.79
 1727.41  245.38 1748.89  249.04 1777.46  249.56  1804.7  252.43 1863.69  254.78
#Mann= 0 , 0 , 0
Bank Sta=1308.04,1347.9
Exp/Cntr=.3,.1

Type RM Length L Ch R = 1 ,44090.86,341.65,247.46,149.74
XS GIS Cut Line= 3
     1838336.041      412217.365     1838742.814      411383.683
     1838698.512      410997.048
#Sta/Elev= 30
       0  244.35    75.7   243.4   92.04  242.41  130.36   238.5  200.97  233.22
  242.66  230.86  289.33  229.01  302.41  228.95  396.01  226.27  447.76  225.79
  462.75  225.94     513  224.73  534.99  224.97  596.18  224.15  676.67  224.12
  732.02  223.32  738.72  223.35   754.2  223.79  769.01  223.77  812.56  224.39
  862.51  228.34  870.93  228.78  898.66  229.35  949.44  230.99  990.12  232.93
 1024.25  233.87 1070.25  235.91 1138.36  238.05 1177.01  240.29 1316.79   246.2
#Mann= 0 , 0 , 0
Bank Sta=738.72,769.01
Exp/Cntr=.3,.1

Type RM Length L Ch R = 1 ,43843.40,491.61,459.01,347.32
XS GIS Cut Line= 3
     1839149.587      412527.479     1838795.171      411266.887
     1838746.841      410980.938
#Sta/Elev= 30
       0  242.23   42.85  240.84   70.75  237.71  101.52  237.51  122.63  236.62
  162.57  236.18  200.58  233.87  223.85  233.35   263.7  231.65  383.71   230.5
  447.98  229.35  515.54  227.32  724.42  225.24  756.84  225.28   796.1  224.35
  834.97  224.55 1028.46  223.43 1032.88  222.78 1062.05  223.31 1084.39  224.34
 1103.67  228.35 1203.87  228.76 1236.47  232.13 1248.08  232.32  1284.4  236.21
  1294.8  236.85 1315.38  237.57  1372.1  238.27 1571.35   245.6 1599.47  246.26
#Mann= 0 , 0 , 0
Bank Sta=1028.46,1062.05
Exp/Cntr=.3,.1

Type RM Length L Ch R = 1 ,43384.39,348.12,413.2,288.36
XS GIS Cut Line= 5
     1839818.144      412177.091     1839741.622      411850.867
     1839568.442      411669.632     1838960.296      411125.926
     1838787.116      410932.608
#Sta/Elev= 30
       0  250.99    64.6   250.7  165.08  248.99  229.97  249.51   271.5  251.48
  314.06  251.25  342.12  249.48  375.16  248.49  390.81  246.08  402.94  245.73
  429.91   243.5  499.06  236.48  545.92  233.24  571.33  232.18  662.44  229.78
  710.28  227.26  798.65  225.14  924.08  223.65 1034.61  223.75 1064.73  223.74
 1091.02  223.45 1131.93  224.41 1152.66  229.07 1189.93  230.55  1247.5  235.37
 1282.55  236.02 1379.46  241.73 1463.59  243.43 1622.28     245 1661.05  246.27
#Mann= 0 , 0 , 0
Bank Sta=1034.61,1064.73
Exp/Cntr=.3,.1

Type RM Length L Ch R = 1 ,42971.19,569.17,672.78,666.05
XS GIS Cut Line= 5
     1840321.575      411746.154     1839874.528       411387.71
      1839302.63      411065.514     1839056.955      410932.608
     1838895.857      410779.565
#Sta/Elev= 30
       0  256.07   57.74  254.13  180.72  252.66  282.85  249.43   311.3  249.17
  420.29  246.29  456.68  243.73  479.74  240.74  525.07  237.15  543.09  236.24
  561.86  233.88  625.88  232.62  701.41  232.25  758.18  230.76  815.69  225.46
  844.03   224.5  983.17  223.02 1014.83  222.84 1016.06  222.86 1202.03  224.49
 1223.24  230.94 1251.22  235.01 1266.44  235.95 1278.68  236.01 1300.34   237.9
 1320.16  238.73 1342.88  238.82 1372.92  239.95  1567.7  241.73 1730.94   245.9
#Mann= 0 , 0 , 0
Bank Sta=983.17,1016.06
Exp/Cntr=.3,.1

Type RM Length L Ch R = 1 ,42298.41,704.41,813.8,756.26
XS GIS Cut Line= 2
     1840469.562      411678.192     1839455.445      410024.199
#Sta/Elev= 30
       0   258.1   99.83   252.6  124.69   249.5  276.49   236.2  560.83  231.36
  677.16  227.98  799.92  226.49  835.08  225.52  854.22  223.81  930.62  222.15
  991.52  222.99 1092.18  222.44 1127.22  222.43 1157.09   222.5 1183.41  225.67
 1206.83  226.39 1367.91  229.49 1406.47  233.06 1470.15  234.73 1477.64  237.77
 1504.41  241.06 1527.03  246.33 1554.84  248.83 1628.41  258.04 1666.94  261.35
 1704.46  262.27 1770.06  261.95 1836.68  259.79 1892.46  256.53 1940.14  256.05
#Mann= 0 , 0 , 0
Bank Sta=1092.18,1127.22
Exp/Cntr=.3,.1

Type RM Length L Ch R = 1 ,41484.61,865.6,1013.71,809.02
XS GIS Cut Line= 2
     1840992.373      411573.629     1840187.434       409501.35
#Sta/Elev= 30
       0  259.76    9.37  257.64   64.43  256.97  128.84   258.9  146.23  261.12
  175.15   262.4  248.11  261.21  297.58  258.24  337.31  252.82  366.71  250.85
  489.99   237.6  610.28  231.15  743.52  229.25   947.7  223.03 1109.29  221.23
 1260.51  221.21 1290.62  221.01 1291.63  221.01 1399.15  221.51 1450.62  223.06
 1470.41  225.75 1486.61  229.73 1513.97  231.12 1559.91  238.08 1651.19  243.43
 1669.39  245.83  1725.2  249.71 1930.11  250.12 2032.41   253.3 2223.12  250.48
#Mann= 0 , 0 , 0
Bank Sta=1260.51,1291.63
Exp/Cntr=.3,.1

Type RM Length L Ch R = 1 ,40470.89,671.26,630.64,565.59
XS GIS Cut Line= 4
     1841740.389       411110.32     1841402.579      410318.882
     1841209.541      409916.719     1840702.816      409289.346
#Sta/Elev= 30
       0  250.09   45.67  250.56   80.09  249.52  128.84  245.93  145.94  243.88
  191.54  240.62  227.98  237.16  274.86  234.46  298.34   232.4   335.5  230.86
  379.86  230.77  392.26  228.31  460.82  226.66  471.76   225.6  508.26  224.45
   818.6  221.06 1079.78  220.36 1109.36  220.07 1356.11  219.74 1424.45  220.82
 1513.21  225.71 1625.01  225.63 1694.67  227.28 1744.83  233.43 1835.53  240.63
 1879.74  245.39 1902.55  245.82 1924.41  248.54  2011.2  252.25 2113.06  251.79
#Mann= 0 , 0 , 0
Bank Sta=1079.78,1109.36
Exp/Cntr=.3,.1

Type RM Length L Ch R = 1 ,39840.25,994.82,997.76,850.49
XS GIS Cut Line= 6
     1842995.803      410699.016     1842838.732      410642.632
     1842552.783      410618.467      1842399.74       410566.11
     1841437.179      409321.628     1841034.434      409007.487
#Sta/Elev= 30
       0  254.06    15.6  254.21  191.82  249.32   322.6  242.97  346.77  242.66
  422.74  238.68  521.62  231.59  573.72  228.76   591.3  228.13  723.18  227.53
  740.13  226.54  759.21  223.67  814.25  222.27 1033.32  220.85 1343.93  221.05
 1695.39  218.81 1725.09  218.29 1735.18  218.22 1860.61  220.07 1880.31  224.22
 1923.72   224.4 1950.42  225.65 1986.24  226.32 2138.32  227.83 2234.72  230.08
 2302.55  230.43 2389.44  232.31 2482.33   236.2  2568.7  234.28 2699.67  236.59
#Mann= 0 , 0 , 0
Bank Sta=1695.39,1725.09
Exp/Cntr=.3,.1

Type RM Length L Ch R = 1 ,38842.49,788.83,819.33,530.65
XS GIS Cut Line= 6
     1843612.003      409490.781     1843450.905      409563.275
     1843112.599      409514.946     1842862.897      409402.177
     1841666.744      408677.236     1841223.724      408681.263
#Sta/Elev= 30
       0  261.64   68.53  262.27  124.59  260.62   265.7  254.14  292.28  252.11
  302.32   250.2  319.99  249.58  499.17  248.99  736.71  233.51  766.51  229.17
  795.59  228.78  819.23  225.42   876.6  224.36  898.96  222.78 1132.33  221.08
  1366.6  221.87 1439.08  220.13 1476.81  217.28 1492.02  217.57 1523.71  218.65
 1597.91  217.86 1667.29  221.81 2084.59   225.1 2120.48   227.1 2168.24   233.4
 2204.97  235.36 2383.48  234.45 2462.11  236.03 2584.48  235.95 2640.74  238.05
#Mann= 0 , 0 , 0
Bank Sta=1492.02,1523.71
Exp/Cntr=.3,.1

Type RM Length L Ch R = 1 ,38023.16,314.24,421.84,413.07
XS GIS Cut Line= 6
     1843519.372      408604.741     1843217.313      408447.671
      1842999.83      408371.149     1842617.222      408487.945
     1841992.967      408524.192     1841219.697      408532.247
#Sta/Elev= 30
       0   258.3  138.29  253.54  196.17  250.35  236.51  250.12  320.65  252.37
  398.64  251.41  469.47  247.86  501.49  244.86  589.58  241.26  621.87  235.74
  723.09  227.76  825.14   224.5 1001.12  220.52 1120.76  219.61 1168.61  217.72
 1379.14  218.24 1409.95  217.24 1421.05  216.91 1499.91  216.96 1538.55  223.16
 1554.71  223.38 1593.61  228.14 1619.96  229.41 1695.05  229.06 1757.11  230.43
 1785.51  232.22 1897.35  233.48 1951.64  235.54 2247.37  234.92 2369.66  237.82
#Mann= 0 , 0 , 0
Bank Sta=1379.14,1409.95
Exp/Cntr=.3,.1

Type RM Length L Ch R = 1 ,37601.33,705.91,684.19,582.36
XS GIS Cut Line= 6
     1843539.509      408560.439      1843048.16       408306.71
     1842758.183      408266.436     1842625.277      408254.353
     1842146.011       408101.31     1841288.163      407819.388
#Sta/Elev= 30
       0  257.94   99.49  255.62  168.92  252.96  341.02  251.73     529  246.89
  674.77  235.03  727.01  233.38   755.1  231.38  800.58  231.54  820.04  230.62
  838.07  227.93  852.25  222.93  979.21  222.16 1027.51  218.84 1072.53  217.24
 1116.05  218.31  1195.1  216.75 1326.23  218.13 1373.93  216.75  1383.7  216.27
 1466.58  217.43 1486.65  223.19 1722.78  224.66 1904.17  222.57 1926.82   223.5
 2001.63  230.27 2086.72  233.32 2269.36  233.62 2352.92   236.9  2385.3  236.94
#Mann= 0 , 0 , 0
Bank Sta=1326.23,1373.93
Exp/Cntr=.3,.1
