--- Barnes Creek.prj (project) ---

Proj Title=Barnes Creek Limited Detail Study
Current Plan=p01
Default Exp/Contr=0.3,0.1
English Units
Geom File=g01
Flow File=f01
Plan File=p01
Y Axis Title=Elevation
X Axis Title(PF)=Main Channel Distance
X Axis Title(XS)=Station
BEGIN DESCRIPTION:
Barnes Creek
END DESCRIPTION:
DSS Export Rating Curves= 0
DSS Export Rating Curve Sorted= 0
DSS Export Volume Flow Curves= 0
DXF OffsetX= 0
DXF OffsetY= 0
DXF ScaleX= 1
DXF ScaleY= 10

--- Barnes Creek.p01 (plan) ---

Plan Title=100-Year Single
Program Version=3.12
Short Identifier=100Year
Geom File=g01
Flow File=f01
Subcritical Flow
K Sum by GR= 0
Std Step Tol= 0.01
Critical Tol= 0.01
Num of Std Step Trials= 20
Max Error Tol= 0.3
Flow Tol Ratio= 0.001
Split Flow NTrial= 30
Split Flow Tol= 0.02
Split Flow Ratio= 0.02
Log Output Level= 0
Friction Slope Method= 1
Unsteady Friction Slope Method= 2
Unsteady Bridges Friction Slope Method= 1
Parabolic Critical Depth
Global Vel Dist= 0 , 0 , 0
Global Log Level= 0
CheckData=True
Encroach Param=-1 ,10,10, 2
Encroach River=Barnes Creek
Encroach Reach=Reach-1
Encroach Node=34090
       1 4962.26 5030.08
Encroach Node=33500
       1    4853  5021.1
Encroach Node=33103
       1    4902 5056.22
Encroach Node=32575
       1    4969    5031
Encroach Node=32482
       1    4974    5026
Encroach Node=31974
       1    4966    5045
Encroach Node=31536
       1  4976.8  5023.2
Encroach Node=31081
       1 4969.04  5023.2
Encroach Node=30786
       1 4965.92  5023.2
Encroach Node=30118
       1  4974.4 5029.04
Encroach Node=29500
       1 4922.97 5084.26
Encroach Node=29000
       1 4940.74  5025.6
Encroach Node=28543
       1 4966.35  5030.3
Encroach Node=27961
       1 4899.48 5211.37
Encroach Node=27458
       1 4769.37  5025.6
Encroach Node=26708
       1  4964.7  5025.6
Encroach Node=26019
       1  4974.4  5025.6
Encroach Node=25596
       1 4883.93 5061.85
Encroach Node=25121
       1  4974.4 5088.82
Encroach Node=24475
       1 4960.65  5026.2
Encroach Node=24040
       1 4966.82 5094.05
Encroach Node=23661
       1 4952.58 5072.67
Encroach Node=23034
       1  4767.5  5032.5
Encroach Node=22928
       1  4767.5  5032.5
Encroach Node=22459
       1  4946.8  5026.5
Encroach Node=21942
       1 4948.12 5077.23
Encroach Node=21560
       1 4939.81  5026.5
Encroach Node=21000
       1  4973.5  5026.5
Encroach Node=20500
       1  4973.5 5058.65
Encroach Node=19878
       1  4973.5  5026.5
Encroach Node=19500
       1  4973.3 5113.92
Encroach Node=18980
       1 4878.59  5026.7
Encroach Node=18521
       1  4973.3 5030.77
Encroach Node=18000
       1  4982.3    5030
Encroach Node=17500
       1  4982.3    5060
Encroach Node=17027
       1  4982.3 5106.94
Encroach Node=16404
       1  4973.3  5026.7
Encroach Node=15907
       1 4965.46  5026.7
Encroach Node=15404
       1 4968.58  5026.7
Encroach Node=14500
       1    4982    5095
Encroach Node=13745
       1    4973    5027
Encroach Node=13365
       1    4973    5027
Encroach Node=12938
       1 4967.54    5027
Encroach Node=12183
       1 4956.53 5031.65
Encroach Node=11689
       1 4972.32 5036.64
Encroach Node=11000
       1    4973 5033.71
Encroach Node=10500
       1    4973    5027
Encroach Node=10000
       1 4969.75 5090.29
Encroach Node=9292
       1    4410    5028
Encroach Node=8862
       1    4960    5070
Encroach Node=8420
       1    4950    5019
Encroach Node=7902
       1    4970    5019
Encroach Node=7404
       1    4972    5028
Encroach Node=7000
       1    4972    5028
Encroach Node=6317
       1 4968.26 5064.22
Encroach Node=5802
       1  4971.7  5028.3
Encroach Node=5231
       1 4969.83  5028.3
Encroach Node=4913
       1  4958.9  5028.3
Encroach Node=4596
       1  4971.7  5028.3
Encroach Node=4172
       1    4970  5018.3
Encroach Node=3808
       1    4963    5037
Encroach Node=3696
       1    4963    5037
Encroach Node=3259
       1 4955.28  5028.3
Encroach Node=2887
       1 4963.48  5018.3
Encroach Node=2500
       1  4971.7  5028.3
Encroach Node=2000
       1 4971.42 5108.82
Encroach Node=1500
       1  4971.7  5028.3
Encroach Node=768
       1 4898.52 5056.12
Encroach Node=171
       1  4955.6 5102.91
BEGIN DESCRIPTION:
100Year Run
END DESCRIPTION:
Computation Interval=1HOUR
Output Interval=1HOUR
Run HTab= 0
Run UNet= 0
Run PostProcess= 0
UNET Theta= 1
UNET Theta Warmup= 1
UNET ZTol= 0.02
UNET ZSATol= 0.05
UNET MxIter= 20
UNET MaxInSteps= 0
UNET DtIC= 0
UNET DtMin= 0
UNET MaxCRTS= 20
UNET WFStab= 2
UNET SFStab= 1
UNET WFX= 1
UNET SFX= 1
UNET DSS MLevel= 4
UNET DZMax Abort= 100
UNET Convert EG Bridges=-1
UNET Use Existing IB Tables=-1
UNET Froude Reduction=False
UNET Froude Limit= 1
UNET Froude Power= 10
Instantaneous Interval=1HOUR
Write IC File= 0
Echo Input=False
Echo Output=False
Write Detailed= 0
Detailed Automatic Start=False, 10

--- Barnes Creek.f01 (steady flow) ---

Flow Title=100-year Single
Program Version=3.12
Number of Profiles= 2
Profile Names=100-year,100-FW
River Rch & RM=Barnes Creek,Reach-1         ,34090
    3458    3458
River Rch & RM=Barnes Creek,Reach-1         ,33103
    4054    4054
River Rch & RM=Barnes Creek,Reach-1         ,30118
    4687    4687
River Rch & RM=Barnes Creek,Reach-1         ,24475
    4838    4838
River Rch & RM=Barnes Creek,Reach-1         ,23034
    4913    4913
River Rch & RM=Barnes Creek,Reach-1         ,19500
    4965    4965
River Rch & RM=Barnes Creek,Reach-1         ,14500
    5040    5040
River Rch & RM=Barnes Creek,Reach-1         ,9292
    5263    5263
River Rch & RM=Barnes Creek,Reach-1         ,6317
    5335    5335
River Rch & RM=Barnes Creek,Reach-1         ,3259
    5348    5348
River Rch & RM=Barnes Creek,Reach-1         ,768
    5452    5452
Boundary for River Rch & Prof#=Barnes Creek,Reach-1         , 1
Up Type= 0
Dn Type= 3
Dn Slope=0.0019
Boundary for River Rch & Prof#=Barnes Creek,Reach-1         , 2
Up Type= 0
Dn Type= 3
Dn Slope=0.0019
DSS Import GetInterval= 0
DSS Import GetPeak= 0
DSS Import FillOption= 0

--- Barnes Creek.g01 (geometry) ---

Geom Title=Existing Conditions
Program Version=3.12

River Reach=Barnes Creek    ,Reach-1
Reach XY= 30
      1721906.27       634266.66      1721997.22       633855.93
      1721681.27       633871.65      1721199.83       632489.62
      1719311.74       632546.69      1719195.41       631469.37
      1717966.35       631039.45      1717232.85       631682.75
      1715978.62       630336.41      1714891.18       630675.28
      1714112.27        630265.6      1713874.55       629193.33
      1713222.09       628854.46      1712802.29       628075.55
      1712195.34       628227.28      1711613.69       627645.63
      1711537.82       628131.18      1710015.41       628611.68
      1709737.23       627023.51       1708396.9        626917.3
      1708310.91       625647.78      1707188.07       623978.69
      1708260.34       622714.22      1706004.53       621935.31
      1706287.77       620018.39      1705063.77       619482.26
      1703450.45       616767.65      1701759.25       615958.57
       1702349.2       614320.75      1701186.84       614324.38

Type RM Length L Ch R = 1 ,34090   ,590,590,590
BEGIN DESCRIPTION:
Barnes Creek 68.0
END DESCRIPTION:
XS GIS Cut Line= 3
      1717405.39       631271.41      1717486.31       631410.49
       1717592.5       631521.74
#Sta/Elev= 10
  4835.4  486.56  4875.4  485.48  4988.9  475.86  4990.4  472.86  5009.6  472.86
  5011.1  475.86  5036.3  478.14  5096.3  486.28  5146.3  496.05  5150.1  496.52
#Mann= 3 ,-1 , 0
  4835.4     .15       0  4988.9     .05       0  5011.1     .15       0
Bank Sta=4988.9,5011.1
Exp/Cntr=0.3,0.1

Type RM Length L Ch R = 1 ,33500   ,397,397,397
BEGIN DESCRIPTION:
Barnes Creek 67.0
END DESCRIPTION:
XS GIS Cut Line= 3
      1717324.52        631359.9      1717076.16       631587.25
      1717018.98       631643.19
#Sta/Elev= 17
  4663.3  483.97  4753.3  479.08  4773.3  478.93  4903.3   473.9  4933.3  474.22
  4943.3  473.52  4983.3  473.23  4988.9  470.27  4990.4  467.27  5009.6  467.27
  5011.1  470.27    5030  476.82    5040  478.03    5050  479.58    5060  481.75
    5070  484.78    5080  490.44
#Mann= 3 ,-1 , 0
  4663.3     .15       0  4988.9     .05       0  5011.1     .14       0
Bank Sta=4988.9,5011.1
Exp/Cntr=0.3,0.1

Type RM Length L Ch R = 1 ,33103   ,528,528,528
BEGIN DESCRIPTION:
Barnes Creek 66.0
END DESCRIPTION:
XS GIS Cut Line= 3
      1716960.43       631124.76      1716841.58       631289.13
      1716735.39       631407.96
#Sta/Elev= 23
  4795.2  491.86  4805.2   490.4  4815.2   488.4  4835.2  483.27  4845.2  479.42
  4865.2  468.96  4875.2  469.68  4935.2  468.92  4945.2   468.5  4955.2  467.72
  4965.2  466.66  4975.2  465.86  4986.8  462.86  4988.3  459.86  5011.7  459.86
  5013.2  462.86    5088  471.74    5108  474.45    5118  476.57    5128  479.39
    5138  483.27    5148  486.77  5157.4  490.37
#Mann= 3 ,-1 , 0
  4795.2     .15       0  4986.8     .05       0  5013.2     .14       0
Bank Sta=4986.8,5013.2
Exp/Cntr=0.5,0.3

Type RM Length L Ch R = 1 ,32575   ,93,93,93
BEGIN DESCRIPTION:
FLINT-HILL-RD-US
END DESCRIPTION:
XS GIS Cut Line= 3
      1716903.32       630954.57      1716430.29       630972.81
      1716218.84       630944.69
#Sta/Elev= 30
  4528.1  481.78  4538.1   478.9  4548.1  476.96  4588.1  471.95  4598.1  470.13
  4608.1  469.22  4648.1  467.13  4728.1  466.48  4768.1  467.31  4808.1  466.25
  4828.1  468.01  4868.1  468.21  4908.1  465.96  4928.1  465.51  4948.1  465.74
  4968.1  463.59    4982   461.4    4984   456.5    5016   456.5    5018   461.4
  5041.5  463.71  5061.5  468.02  5101.5  474.76  5111.5  474.85  5131.5  477.95
  5151.5  478.97  5161.5  480.41  5171.5  481.12  5191.5  481.54  5214.8  482.96
#Mann= 3 ,-1 , 0
  4528.1     .15       0    4982     .05       0    5018     .15       0
#XS Ineff= 2 , 0
       0    4969   471.2    5031       0  471.03
Permanent Ineff=
       F       F
Bank Sta=4982,5018
Exp/Cntr=0.5,0.3

Type RM Length L Ch R = 3 ,32531   ,,,
BEGIN DESCRIPTION:
FLINT-HILL-RD-TOR
Structure ID: LDS_BAC_03
Approximate Survey Structure
END DESCRIPTION:
Bridge Culvert--1,0,-1,-1, 0
Deck Dist Width WeirC Skew NumUp NumDn MinLoCord MaxHiCord MaxSubmerge Is_Ogee
33.5,21,3,0, 17, 17, , , 0.95, 0, 1,1,,
    4530    4550    4560    4570  4579.4    4979    4979    5021    5021  5050.3
  5101.3  5111.3  5141.3  5151.3  5191.3  5201.3  5205.1
  484.07  477.54   474.9  472.61   471.2   471.2   471.2   471.2   471.2   471.2
  473.75  474.69  476.25  476.34  478.15  479.11  479.22
   436.5   436.5   436.5   436.5   436.5   436.5   469.1   469.1   436.5   436.5
   436.5   436.5   436.5   436.5   436.5   436.5   436.5
    4530    4550    4560    4570  4579.4    4979    4979    5021    5021  5050.3
  5101.3  5111.3  5141.3  5151.3  5191.3  5201.3  5205.1
  484.07  477.54   474.9  472.61   471.2   471.2   471.2   471.2   471.2   471.2
  473.75  474.69  476.25  476.34  478.15  479.11  479.22
   436.5   436.5   436.5   436.5   436.5   436.5   469.1   469.1   436.5   436.5
   436.5   436.5   436.5   436.5   436.5   436.5   436.5
BR Coef= 1 , 1 , 0 ,1.25, 0 ,,,0.8,0,2,0,
WSPro=,,,, 1 ,,,, 0 ,,,, 0 ,,,,-1 ,-1 ,-1 , 0 , 0 , 0 , 0 , 0
BC Design=,, 0 ,, 0 ,,,,,,
BC HTab HWMax=483.07

Type RM Length L Ch R = 1 ,32482   ,508,508,508
BEGIN DESCRIPTION:
FLINT-HILL-RD-DS
END DESCRIPTION:
XS GIS Cut Line= 3
      1716864.38       630881.61      1716415.09       630883.19
      1716221.11       630857.28
#Sta/Elev= 30
  4550.8   483.8  4570.8  477.46  4580.8  473.64  4590.8  470.83  4600.8  468.83
  4630.8  466.91  4650.8  466.63  4680.8  467.68  4740.8  466.94  4780.8  465.33
  4790.8  465.29  4850.8  467.19  4900.8  467.73  4910.8  466.75  4920.8  464.57
  4940.8  464.01  4960.8  464.06  4970.8  462.94  4980.8  460.64    4982  461.15
    4984  456.25    5016  456.25    5018  461.15  5020.1  458.05  5040.1  462.25
  5080.1  465.69  5120.1  471.13  5130.1  472.08  5160.1  476.45  5195.8  479.49
#Mann= 3 ,-1 , 0
  4550.8     .15       0    4982     .05       0    5018     .15       0
#XS Ineff= 2 , 0
       0    4969  470.91    5031       0  470.81
Permanent Ineff=
       F       F
Bank Sta=4982,5018
Exp/Cntr=0.5,0.3

Type RM Length L Ch R = 1 ,31974   ,438,438,438
BEGIN DESCRIPTION:
Barnes Creek 64.0
END DESCRIPTION:
XS GIS Cut Line= 3
      1716225.54       630409.06      1716122.19       630497.21
       1716003.6       630609.72
#Sta/Elev= 19
  4864.2   496.4  4874.2  489.07  4884.2   482.3  4894.2  478.78  4904.2  474.15
  4914.2  469.86  4924.2  466.97  4964.2  457.66  4974.2  458.51  4984.2  457.89
  4986.8  455.97  4988.3  452.97  5011.7  452.97  5013.2  455.97    5050  459.69
    5080  467.51    5130   474.4    5140  475.19  5163.5  476.09
#Mann= 3 ,-1 , 0
  4864.2     .15       0  4986.8     .05       0  5013.2     .15       0
Bank Sta=4986.8,5013.2
Exp/Cntr=0.3,0.1

Type RM Length L Ch R = 1 ,31536   ,455,455,455
BEGIN DESCRIPTION:
Barnes Creek 63.0
END DESCRIPTION:
XS GIS Cut Line= 3
      1715745.24       630299.61      1715777.15       630390.81
        1715879.       630606.67
#Sta/Elev= 23
  4899.9  480.84  4919.9   473.7  4939.9  466.06  4969.9  456.64  4979.9  456.46
  4986.8  453.12  4988.3  450.12  5011.7  450.12  5013.2  453.12  5016.5  455.47
  5026.5  458.53  5046.5  460.37  5056.5  461.86  5066.5  462.86  5076.5  463.26
  5116.5  463.93  5126.5  464.94  5156.5  465.72  5166.5  466.37  5176.5   467.5
  5206.5  469.11  5216.5  470.27  5235.2  471.48
#Mann= 3 ,-1 , 0
  4899.9     .15       0  4986.8     .05       0  5013.2     .15       0
Bank Sta=4986.8,5013.2
Exp/Cntr=0.3,0.1

Type RM Length L Ch R = 1 ,31081   ,295,295,295
BEGIN DESCRIPTION:
Barnes Creek 62.0
END DESCRIPTION:
XS GIS Cut Line= 3
      1715386.52       630337.56      1715365.24       630567.13
      1715363.72       630646.16
#Sta/Elev= 13
  4769.9  466.49  4779.9  465.97  4949.9  453.01  4986.8  448.23  4988.3  445.23
  5011.7  445.23  5013.2  448.23  5020.4  452.97  5030.4  459.05  5040.4  465.42
  5050.4  471.48  5060.4  476.44  5079.5  484.83
#Mann= 3 ,-1 , 0
  4769.9     .15       0  4986.8     .05       0  5013.2     .15       0
Bank Sta=4986.8,5013.2
Exp/Cntr=0.3,0.1

Type RM Length L Ch R = 1 ,30786   ,668,668,668
BEGIN DESCRIPTION:
Barnes Creek 61.0
END DESCRIPTION:
XS GIS Cut Line= 3
      1715049.09       630436.41        1715081.       630589.93
      1715108.36       630671.99
#Sta/Elev= 20
  4842.1  474.55  4852.1  469.78  4862.1  464.62  4882.1  457.66  4892.1  455.97
  4912.1  453.28  4962.1  450.79  4982.1  448.77  4986.8  447.16  4988.3  444.16
  5011.7  444.16  5013.2  447.16  5018.9  450.05  5028.9  459.28  5038.9  462.44
  5048.9   464.2  5058.9  465.59  5068.9  466.41  5078.9  467.82  5085.4  468.38
#Mann= 3 ,-1 , 0
  4842.1     .15       0  4986.8     .05       0  5013.2     .15       0
Bank Sta=4986.8,5013.2
Exp/Cntr=0.3,0.1

Type RM Length L Ch R = 1 ,30118   ,618,618,618
BEGIN DESCRIPTION:
Barnes Creek 60.0
END DESCRIPTION:
XS GIS Cut Line= 3
      1714731.08       630306.77      1714685.95       630382.78
      1714443.71       630931.38
#Sta/Elev= 29
  4907.5  461.08  4917.5   458.8  4927.5     457  4947.5  454.76  4967.5  449.89
  4984.4  443.59  4985.9  440.59  5014.1  440.59  5015.6  443.59  5065.9  449.78
  5075.9  451.74  5085.9  451.23  5095.9  452.04  5105.9  453.32  5115.9  454.07
  5185.9  454.47  5195.9  455.09  5225.9  455.88  5235.9   455.5  5245.9  454.86
  5345.9   453.1  5455.9  453.15  5495.9  454.81  5535.9   459.1  5545.9   461.2
  5555.9  463.61  5575.9  468.79  5585.9  471.96  5595.6  475.39
#Mann= 3 ,-1 , 0
  4907.5     .15       0  4984.4    .045       0  5015.6     .13       0
Bank Sta=4984.4,5015.6
Exp/Cntr=0.3,0.1

Type RM Length L Ch R = 1 ,29500   ,500,500,500
BEGIN DESCRIPTION:
Barnes Creek 59.0
END DESCRIPTION:
XS GIS Cut Line= 3
      1714341.55       630088.31      1714106.73        630257.3
      1713997.19       630347.18
#Sta/Elev= 27
  4710.7  465.78  4750.7  459.62  4760.7  457.27  4780.7  454.22  4790.7  452.26
  4800.7  451.04  4810.7  450.25  4820.7  449.95  4830.7  450.59  4860.7  450.67
  4890.7  449.45  4900.7  446.73  4910.7  445.86  4960.7   447.1  4980.7  446.11
  4984.4  441.02  4985.9  438.02  5014.1  438.02  5015.6  441.02    5020  445.27
    5060  442.75    5090  442.39    5100  446.34    5110  456.39    5120  462.35
    5130  469.04  5141.7  475.97
#Mann= 3 ,-1 , 0
  4710.7     .13       0  4984.4    .045       0  5015.6     .13       0
Bank Sta=4984.4,5015.6
Exp/Cntr=0.3,0.1

Type RM Length L Ch R = 1 ,29000   ,457,457,457
BEGIN DESCRIPTION:
Barnes Creek 58.0
END DESCRIPTION:
XS GIS Cut Line= 3
      1714187.21       629708.29      1713870.37       629820.75
      1713771.56       629872.18
#Sta/Elev= 26
  4663.8  464.36  4743.8  453.15  4753.8  452.22  4763.8   452.3  4773.8  451.95
  4793.8  450.05  4803.8  449.58  4873.8  448.92  4883.8  447.56  4893.8  445.87
  4903.8  444.89  4913.8  444.17  4923.8  443.91  4963.8  439.89  4984.4  438.79
  4985.9  435.79  5014.1  435.79  5015.6  438.79    5020   448.4    5030  451.17
    5060  456.21    5070  458.42    5090  464.11    5100  467.34    5110  470.93
  5111.4  471.33
#Mann= 3 ,-1 , 0
  4663.8     .13       0  4984.4    .045       0  5015.6     .13       0
Bank Sta=4984.4,5015.6
Exp/Cntr=0.3,0.1

Type RM Length L Ch R = 1 ,28543   ,582,582,582
BEGIN DESCRIPTION:
Barnes Creek 57.0
END DESCRIPTION:
XS GIS Cut Line= 3
      1714125.49       629387.67      1713849.96       629373.42
      1713567.37       629439.91
#Sta/Elev= 30
  4727.5  466.88  4747.5  464.67  4757.5  463.87  4767.5  462.63  4787.5  459.55
  4827.5  451.72  4847.5  449.47  4857.5  448.76  4867.5  448.86  4907.5  449.08
  4927.5  446.28  4947.5  445.17  4967.5  439.67  4984.4  437.98  4985.9  434.98
  5014.1  434.98  5015.6  437.98  5023.4  443.16  5053.4  447.72  5063.4  448.48
  5103.4  449.09  5113.4  448.63  5163.4  447.87  5223.4  448.35  5243.4  452.95
  5253.4  455.58  5273.4  462.53  5283.4  464.58  5293.4  467.29  5293.7  467.37
#Mann= 3 ,-1 , 0
  4727.5     .15       0  4984.4     .05       0  5015.6     .15       0
Bank Sta=4984.4,5015.6
Exp/Cntr=0.3,0.1

Type RM Length L Ch R = 1 ,27961   ,503,503,503
BEGIN DESCRIPTION:
Barnes Creek 56.0
END DESCRIPTION:
XS GIS Cut Line= 3
      1713762.09       628829.55      1713581.59       628943.55
      1713251.47       629202.42
#Sta/Elev= 30
    4791  462.92    4801  461.11    4811  460.17    4821  458.44    4831  455.33
    4861  446.78    4881  439.95    4901  444.39    4911   445.3    4921  445.25
    4931  445.92    4961  445.17  4984.4  436.41  4985.9  433.41  5014.1  433.41
  5015.6  436.41  5034.5  445.93  5094.5  447.29  5114.5  446.91  5134.5  446.96
  5204.5  444.12  5224.5  444.56  5234.5  445.07  5244.5  445.12  5284.5  446.55
  5294.5  445.36  5304.5  450.03  5314.5  453.31  5324.5  454.58    5424   463.5
#Mann= 3 ,-1 , 0
    4791     .15       0  4984.4     .05       0  5015.6     .15       0
Bank Sta=4984.4,5015.6
Exp/Cntr=0.3,0.1

Type RM Length L Ch R = 1 ,27458   ,750,750,750
BEGIN DESCRIPTION:
Barnes Creek 55.0
END DESCRIPTION:
XS GIS Cut Line= 3
       1713427.2       628378.33      1713149.35        628758.3
      1713037.71       628964.95
#Sta/Elev= 30
  4529.8  471.09  4549.8  467.18  4569.8  462.21  4599.8   452.7  4609.8  449.93
  4629.8  445.78  4639.8  444.89  4729.8   444.5  4749.8  444.02  4899.8  445.22
  4949.8     443  4969.8   439.2  4984.4  435.01  4985.9  432.01  5014.1  432.01
  5015.6  435.01  5020.5  442.43  5030.5  444.07  5040.5  445.26  5050.5  445.28
  5060.5  445.82  5070.5  446.92  5100.5  453.32  5110.5  454.15  5140.5  457.76
  5150.5  458.47  5160.5  458.78  5180.5  460.11  5220.5  461.42  5235.4  461.51
#Mann= 3 ,-1 , 0
  4529.8     .15       0  4984.4     .05       0  5015.6     .15       0
Bank Sta=4984.4,5015.6
Exp/Cntr=0.3,0.1

Type RM Length L Ch R = 1 ,26708   ,689,689,689
BEGIN DESCRIPTION:
Barnes Creek 54.0
END DESCRIPTION:
XS GIS Cut Line= 3
      1712874.95       628001.81      1712836.41       628094.31
      1712603.89       628926.74
#Sta/Elev= 30
    4897  459.61    4907  452.51    4917   447.2    4927  442.96    4967  438.18
  4984.4  434.77  4985.9  431.77  5014.1  431.77  5015.6  434.77  5027.2  445.33
  5047.2  444.32  5057.2  444.43  5077.2  446.53  5097.2  443.84  5107.2  443.49
  5147.2  443.62  5187.2  442.69  5237.2  443.55  5337.2  441.87  5447.2  442.18
  5467.2  441.66  5537.2  442.19  5607.2   446.7  5617.2  446.63  5657.2  448.53
  5687.2  451.05  5717.2  450.89  5727.2  450.12  5837.2   455.4  5861.5  457.09
#Mann= 4 ,-1 , 0
    4897     .15       0  4984.4     .05       0  5015.6     .15       0
  5077.2      10       0
Bank Sta=4984.4,5015.6
Exp/Cntr=0.3,0.1

Type RM Length L Ch R = 1 ,26019   ,423,423,423
BEGIN DESCRIPTION:
Barnes Creek 52.0
END DESCRIPTION:
XS GIS Cut Line= 3
      1712230.25       628152.67      1712187.49       628221.56
      1712065.94       628404.95
#Sta/Elev= 15
  4917.3  451.86  4927.3  449.59  4937.3  446.82  4947.3  442.06  4957.3  439.08
  4984.4  431.84  4985.9  428.84  5014.1  428.84  5015.6  431.84  5018.4   441.6
  5048.4  442.07  5108.4  444.72  5128.4  446.27  5138.4  447.54  5218.4   463.9
#Mann= 3 ,-1 , 0
  4917.3     .15       0  4984.4     .05       0  5015.6     .15       0
Bank Sta=4984.4,5015.6
Exp/Cntr=0.3,0.1

Type RM Length L Ch R = 1 ,25596   ,475,475,475
BEGIN DESCRIPTION:
Barnes Creek 51.0
END DESCRIPTION:
XS GIS Cut Line= 3
      1712201.73       627575.58      1711904.87       627917.56
       1711807.5       628212.02
#Sta/Elev= 30
  4542.7   468.8  4562.7  462.75  4602.7  446.61  4612.7  445.02  4622.7  444.16
  4712.7  441.91  4732.7  440.75  4852.7  439.58  4882.7  440.12  4922.7   439.7
  4942.7  438.71  4952.7  438.56  4982.7  435.82  4984.4  432.61  4985.9  429.61
  5014.1  429.61  5015.6  432.61  5025.6  438.37  5055.6  439.87  5065.6  441.06
  5075.6  440.48  5105.6  440.04  5115.6  438.98  5125.6  438.28  5135.6   438.2
  5225.6  444.53  5245.6  447.48  5275.6   453.5  5285.6  455.95  5305.7  458.46
#Mann= 3 ,-1 , 0
  4542.7     .15       0  4984.4     .05       0  5015.6     .15       0
Bank Sta=4984.4,5015.6
Exp/Cntr=0.3,0.1

Type RM Length L Ch R = 1 ,25121   ,646,646,646
BEGIN DESCRIPTION:
Barnes Creek 50.0
END DESCRIPTION:
XS GIS Cut Line= 3
      1711493.98       627433.02      1711569.99       627663.44
      1711752.87       628223.93
#Sta/Elev= 30
    4757  463.16    4767  460.84    4787  454.83    4797  453.46    4807  452.86
    4817  451.47    4827  448.83    4837   444.1    4847  442.94    4937  439.58
    4977  439.74  4984.4  430.79  4985.9  427.79  5014.1  427.79  5015.6  430.79
  5029.6  433.43  5059.6  431.77  5069.6  431.68  5119.6  438.25  5169.6  440.52
  5189.6  439.86  5259.6  438.74  5459.6  438.63  5469.6   438.9  5479.6  439.46
  5519.6  446.45  5549.6  453.24  5559.6  455.02  5569.6  456.41  5589.2   457.5
#Mann= 3 ,-1 , 0
    4757     .15       0  4984.4     .05       0  5015.6     .15       0
Bank Sta=4984.4,5015.6
Exp/Cntr=0.3,0.1

Type RM Length L Ch R = 1 ,24475   ,435,435,435
BEGIN DESCRIPTION:
Barnes Creek 49.0
END DESCRIPTION:
XS GIS Cut Line= 3
      1711180.51       627504.35      1711403.75       628150.31
      1711455.99       628316.55
#Sta/Elev= 30
  4315.4  466.63  4335.4  459.65  4345.4  453.92  4355.4  451.96  4375.4  451.43
  4395.4  443.44  4405.4  442.13  4425.4  440.84  4475.4  439.93  4545.4  437.36
  4605.4  438.46  4625.4   438.2  4655.4  439.75  4735.4  442.08  4765.4  441.85
  4815.4  438.57  4925.4  436.27  4935.4  435.26  4955.4  431.72  4983.8  428.57
  4985.3  425.57  5014.7  425.57  5016.2  428.57  5018.8  431.19  5028.8  432.21
  5048.8  436.96  5058.8   438.7  5098.8  444.05  5158.8  449.57  5173.1  451.81
#Mann= 4 ,-1 , 0
  4315.4      10       0  4735.4     .15       0  4983.8     .05       0
  5016.2     .15       0
Bank Sta=4983.8,5016.2
Exp/Cntr=0.3,0.1

Type RM Length L Ch R = 1 ,24040   ,379,379,379
BEGIN DESCRIPTION:
Barnes Creek 48.0
END DESCRIPTION:
XS GIS Cut Line= 3
      1710893.15       628048.22       1710990.5       628250.06
      1711232.75       628691.81
#Sta/Elev= 30
  4778.1  454.49  4798.1  452.87  4808.1  451.58  4818.1  450.94  4828.1  450.81
  4848.1  447.13  4858.1  445.86  4868.1  444.89  4878.1  442.99  4908.1  438.32
  4983.8  427.56  4985.3  424.56  5014.7  424.56  5016.2  427.56  5072.2  433.58
  5092.2  434.78  5102.2  435.11  5122.2  434.76  5252.2  436.47  5282.2  436.14
  5362.2  437.06  5392.2  438.19  5422.2  438.99  5432.2  439.93  5442.2  441.53
  5452.2  443.47  5482.2  452.38  5492.2  456.77  5502.2   461.5    5506  463.17
#Mann= 3 ,-1 , 0
  4778.1     .13       0  4983.8     .05       0  5016.2     .15       0
Bank Sta=4983.8,5016.2
Exp/Cntr=0.3,0.1

Type RM Length L Ch R = 1 ,23661   ,627,627,627
BEGIN DESCRIPTION:
Barnes Creek 47.0
END DESCRIPTION:
XS GIS Cut Line= 3
      1710658.01       628212.06      1710665.13       628440.06
      1710824.27       628774.96
#Sta/Elev= 26
    4769  442.81    4779  442.76    4809  441.69    4829  437.94    4839  436.53
    4869  435.47    4909   433.2    4929  432.95    4939   431.5    4949  429.71
  4983.8   426.7  4985.3   423.7  5014.7   423.7  5016.2   426.7  5107.1  434.69
  5117.1  434.98  5157.1  435.25  5177.1  434.38  5187.1  434.37  5257.1  435.11
  5287.1   436.8  5297.1  438.59  5307.1  442.47  5347.1  459.82  5367.1  466.72
  5367.9  466.91
#Mann= 3 ,-1 , 0
    4769     .15       0  4983.8     .05       0  5016.2     .15       0
Bank Sta=4983.8,5016.2
Exp/Cntr=0.5,0.3

Type RM Length L Ch R = 1 ,23034   ,106,106,106
BEGIN DESCRIPTION:
SR-1134-US
END DESCRIPTION:
XS GIS Cut Line= 3
        1710565.       628148.17      1710135.38       628679.17
      1710008.73       628828.31
#Sta/Elev= 30
  4319.2   444.2  4359.2  444.07  4369.2  442.96  4389.2  437.24  4399.2  436.15
  4489.2  433.94  4539.2  434.71  4649.2  432.23  4699.2  434.06  4709.2  433.82
  4729.2  431.91  4739.2  430.18  4759.2  429.89  4769.2   430.5  4839.2  431.42
  4869.2  428.78  4879.2  428.74  4899.2  430.55  4977.5   427.4    4982   422.4
    5018   422.4  5022.5   427.4  5042.2  431.58  5052.2  431.27  5072.2  432.82
  5092.2   436.1  5132.2  450.33  5142.2  452.38  5172.2  453.99  5197.9  456.58
#Mann= 3 ,-1 , 0
  4319.2     .13       0  4977.5     .05       0  5022.5     .15       0
#XS Ineff= 2 , 0
       0  4943.5  435.45  5056.5       0  437.99
Permanent Ineff=
       F       F
Bank Sta=4977.5,5022.5
Exp/Cntr=0.5,0.3

Type RM Length L Ch R = 3 ,22979   ,,,
BEGIN DESCRIPTION:
SR-1134-TOR
Structure ID: LDS_BAC_02
Approximate Survey Structure
END DESCRIPTION:
Bridge Culvert--1,0,-1,-1, 0
Deck Dist Width WeirC Skew NumUp NumDn MinLoCord MaxHiCord MaxSubmerge Is_Ogee
44.5,21,3,0, 25, 25, , , 0.95, 0, 1,1,,
  4321.3  4331.3  4361.3  4421.3  4431.3  4461.3  4481.3  4511.3  4661.3  4711.3
  4731.3  4741.3  4791.3  4801.3  4953.5  4953.5  5046.5  5046.5  5088.8  5098.8
  5108.8  5128.8  5138.8  5188.8  5198.3
   440.7  440.16  439.75   436.9  436.99   436.7  435.97  435.43  436.44  436.16
  436.63  436.33  436.57  436.94   437.6   437.6   437.6   437.6  440.31   440.9
  442.05  443.59  444.79  449.59  450.16
   402.4   402.4   402.4   402.4   402.4   402.4   402.4   402.4   402.4   402.4
   402.4   402.4   402.4   402.4   402.4   435.7   435.7   402.4   402.4   402.4
   402.4   402.4   402.4   402.4   402.4
  4321.3  4331.3  4361.3  4421.3  4431.3  4461.3  4481.3  4511.3  4661.3  4711.3
  4731.3  4741.3  4791.3  4801.3  4953.5  4953.5  5046.5  5046.5  5088.8  5098.8
  5108.8  5128.8  5138.8  5188.8  5198.3
   440.7  440.16  439.75   436.9  436.99   436.7  435.97  435.43  436.44  436.16
  436.63  436.33  436.57  436.94   437.6   437.6   437.6   437.6  440.31   440.9
  442.05  443.59  444.79  449.59  450.16
   402.4   402.4   402.4   402.4   402.4   402.4   402.4   402.4   402.4   402.4
   402.4   402.4   402.4   402.4   402.4   435.7   435.7   402.4   402.4   402.4
   402.4   402.4   402.4   402.4   402.4
Pier Skew, UpSta & Num, DnSta & Num=  ,4976.8, 2 ,4976.8, 2 , 0 , 0 , 0 ,0,0
       1       1
  427.43   435.7
       1       1
   427.3   435.7
Pier Skew, UpSta & Num, DnSta & Num=  ,5023.3, 2 ,5023.3, 2 , 0 , 0 , 0 ,0,0
       1       1
  427.59   435.7
       1       1
  427.56   435.7
BR Coef= 1 , 1 , 0 ,1.25, 0 ,,,0.8,0,2,0,
WSPro=,,,, 1 ,,,, 0 ,,,, 0 ,,,,-1 ,-1 ,-1 , 0 , 0 , 0 , 0 , 0
BC Design=,, 0 ,, 0 ,,,,,,
BC HTab HWMax=456.58

Type RM Length L Ch R = 1 ,22928   ,469,469,469
BEGIN DESCRIPTION:
SR-1134-DS
END DESCRIPTION:
XS GIS Cut Line= 3
      1710420.06       628096.78      1710042.59       628629.68
      1709919.89       628778.08
#Sta/Elev= 30
  4347.3  442.61  4367.3  442.15  4387.3  440.71  4457.3  434.51  4507.3  433.17
  4597.3  432.38  4627.3  431.41  4647.3  432.97  4707.3  433.02  4777.3  434.66
  4817.3  434.11  4877.3  430.06  4917.3  430.78  4947.3  429.08  4957.3  429.69
  4967.3  429.39  4977.5  427.15    4982  422.15    5018  422.15  5022.5  427.15
  5040.3  436.36  5070.3  434.12  5080.3  436.62  5090.3  440.65  5100.3  447.06
  5110.3  450.97  5120.3   457.2  5140.3  460.89  5160.3  463.31  5192.9  465.67
#Mann= 3 ,-1 , 0
  4347.3     .13       0  4977.5     .05       0  5022.5     .15       0
#XS Ineff= 2 , 0
       0  4943.5  432.71  5056.5       0  437.96
Permanent Ineff=
       F       F
Bank Sta=4977.5,5022.5
Exp/Cntr=0.5,0.3

Type RM Length L Ch R = 1 ,22459   ,517,517,517
BEGIN DESCRIPTION:
Barnes Creek 45.0
END DESCRIPTION:
XS GIS Cut Line= 3
      1710229.98       628050.19      1709942.23       628187.49
      1709821.03       628254.66
#Sta/Elev= 25
  4680.2  440.47  4720.2  440.53  4740.2  439.97  4760.2  438.58  4780.2  436.37
  4790.2  435.67  4820.2  432.17  4830.2  431.73  4840.2  430.66  4850.2  430.66
  4910.2  428.69  4940.2  428.88  4960.2   427.7  4970.2   427.6  4980.2  426.39
  4983.5  421.65    4985  418.65    5015  418.65  5016.5  421.65    5019  426.96
    5059  433.34    5069  435.55    5109  447.28    5129  452.22  5137.6  453.56
#Mann= 3 ,-1 , 0
  4680.2     .13       0  4983.5     .05       0  5016.5     .15       0
Bank Sta=4983.5,5016.5
Exp/Cntr=0.3,0.1

Type RM Length L Ch R = 1 ,21942   ,382,382,382
BEGIN DESCRIPTION:
Barnes Creek 44.0
END DESCRIPTION:
XS GIS Cut Line= 3
      1710114.61       627595.86      1709800.53        627702.5
      1709394.45       627905.55
#Sta/Elev= 30
  4671.1  455.18  4691.1  452.03  4701.1  450.05  4721.1  444.93  4761.1  433.82
  4781.1  431.45  4791.1  430.92  4801.1  429.47  4811.1  428.83  4841.1  428.14
  4941.1  429.65  4951.1  429.39  4961.1  428.41  4971.1  427.92  4981.1   425.7
  4983.5  420.11    4985  417.11    5015  417.11  5016.5  420.11  5022.8  424.46
  5082.8  428.92  5132.8  427.73  5182.8  428.58  5232.8  432.28  5252.8  432.73
  5302.8   435.9  5322.8  436.39  5352.8  436.36  5402.8  437.03  5456.8  440.08
#Mann= 3 ,-1 , 0
  4671.1     .15       0  4983.5     .05       0  5016.5     .15       0
Bank Sta=4983.5,5016.5
Exp/Cntr=0.3,0.1

Type RM Length L Ch R = 1 ,21560   ,560,560,560
BEGIN DESCRIPTION:
Barnes Creek 43.0
END DESCRIPTION:
XS GIS Cut Line= 3
      1709950.05       627228.67      1709714.53       627340.04
      1709274.46       627608.47
#Sta/Elev= 30
  4742.2  462.13  4752.2   453.3  4762.2  446.95  4772.2  441.01  4782.2  433.45
  4792.2  429.49  4802.2     428  4812.2  427.92  4832.2  428.24  4852.2  426.88
  4902.2  427.24  4952.2  424.46  4962.2  423.22  4982.2   421.7  4983.5  419.38
    4985  416.38    5015  416.38  5016.5  419.38  5052.7  427.43  5072.7  428.43
  5122.7  429.02  5162.7  430.29  5202.7  428.68  5302.7  429.64  5322.7  429.21
  5332.7  429.41  5462.7  434.28  5472.7  435.47  5502.7  436.59  5518.2  436.78
#Mann= 4 ,-1 , 0
  4742.2     .15       0  4983.5     .05       0  5016.5     .15       0
  5162.7      10       0
Bank Sta=4983.5,5016.5
Exp/Cntr=0.3,0.1

Type RM Length L Ch R = 1 ,21000   ,500,500,500
BEGIN DESCRIPTION:
Barnes Creek 42.0
END DESCRIPTION:
XS GIS Cut Line= 3
      1709603.16       626817.78      1709567.26       626876.82
      1709082.73       627487.95
#Sta/Elev= 24
  4930.9  453.22  4940.9  447.78  4950.9  438.09  4960.9   429.8  4983.5  415.95
    4985  412.95    5015  412.95  5016.5  415.95    5020   426.3    5030  425.38
    5040  424.98    5060  425.59    5090  425.87    5100  425.58    5130  426.36
    5140  426.03    5200  427.52    5460  426.91    5470  427.39    5540   428.6
    5550  430.19    5630  435.61    5670  436.96  5779.9  438.16
#Mann= 3 ,-1 , 0
  4930.9     .15       0  4983.5     .05       0  5016.5     .15       0
Bank Sta=4983.5,5016.5
Exp/Cntr=0.3,0.1

Type RM Length L Ch R = 1 ,20500   ,622,622,622
BEGIN DESCRIPTION:
Barnes Creek 41.0
END DESCRIPTION:
XS GIS Cut Line= 3
      1709113.78       626646.12      1709090.15       626767.44
      1708949.43       627451.41
#Sta/Elev= 23
  4876.4     441  4896.4  433.37  4916.4     427  4926.4  424.26  4936.4  422.95
  4956.4  421.62  4983.5  414.86    4985  411.86    5015  411.86  5016.5  414.86
    5020  422.84    5030  424.31    5050  424.79    5290  423.55    5380  425.61
    5510  433.72    5610  434.46    5640  435.75    5650  435.82    5660  435.58
    5670  434.98    5690  435.74  5698.3  436.28
#Mann= 3 ,-1 , 0
  4876.4     .15       0  4983.5     .05       0  5016.5     .11       0
Bank Sta=4983.5,5016.5
Exp/Cntr=0.3,0.1

Type RM Length L Ch R = 1 ,19878   ,378,378,378
BEGIN DESCRIPTION:
Barnes Creek 40.0
END DESCRIPTION:
XS GIS Cut Line= 3
      1708754.05        626531.1      1708556.84       626998.58
      1708509.36       627117.26
#Sta/Elev= 30
    4493  441.24    4503  440.78    4523  439.25    4553  436.39    4573  433.36
    4583  432.23    4593  431.42    4623  430.25    4653  430.13    4703   428.9
    4733   426.3    4803  421.77    4853  421.57    4873  422.15    4953  418.89
    4963  418.42    4983  418.61  4983.5  412.72    4985  409.72    5015  409.72
  5016.5  412.72  5020.4  418.37  5050.4  414.55  5060.4  417.78  5070.4  421.97
  5080.4  427.72  5100.4  437.87  5110.4  442.36  5120.4  446.43  5128.2  450.09
#Mann= 3 ,-1 , 0
    4493     .15       0  4983.5     .05       0  5016.5     .15       0
Bank Sta=4983.5,5016.5
Exp/Cntr=0.3,0.1

Type RM Length L Ch R = 1 ,19500   ,520,520,520
BEGIN DESCRIPTION:
Barnes Creek 39.0
END DESCRIPTION:
XS GIS Cut Line= 3
      1708544.09       626715.54      1708326.56       626744.07
      1708047.41       626721.03
#Sta/Elev= 26
  4780.6  430.81  4810.6  429.44  4870.6  423.37  4880.6  422.78  4890.6  421.62
  4910.6  418.71  4920.6  417.93  4950.6  417.44  4960.6  417.03  4983.3  412.06
  4984.8  409.06  5015.2  409.06  5016.7  412.06    5030  414.68    5040  415.04
    5060  413.58    5150   413.7    5180  416.67    5190  417.99    5200  422.12
    5220  429.63    5230  435.05    5240   439.4    5250  442.92    5260  445.89
  5280.1  452.31
#Mann= 3 ,-1 , 0
  4780.6     .15       0  4983.3     .05       0  5016.7     .15       0
Bank Sta=4983.3,5016.7
Exp/Cntr=0.3,0.1

Type RM Length L Ch R = 1 ,18980   ,459,459,459
BEGIN DESCRIPTION:
Barnes Creek 38.0
END DESCRIPTION:
XS GIS Cut Line= 3
      1708659.09       626222.52      1708418.06       626237.13
      1708206.24        626235.3
#Sta/Elev= 24
  4757.6  437.75  4767.6  435.82  4787.6  432.38  4817.6  426.24  4827.6  423.58
  4847.6  414.85  4857.6  412.24  4867.6  410.51  4877.6  409.22  4897.6  408.68
  4917.6  409.04  4967.6  412.56  4977.6  412.45  4983.3  407.04  4984.8  404.04
  5015.2  404.04  5016.7  407.04  5019.1  414.39  5039.1  413.84  5089.1  413.98
  5109.1  415.55  5139.1  419.59  5149.1  421.26  5210.9  434.99
#Mann= 3 ,-1 , 0
  4757.6     .15       0  4983.3     .05       0  5016.7     .15       0
Bank Sta=4983.3,5016.7
Exp/Cntr=0.3,0.1

Type RM Length L Ch R = 1 ,18521   ,521,521,521
BEGIN DESCRIPTION:
Barnes Creek 37.0
END DESCRIPTION:
XS GIS Cut Line= 3
      1708525.01         625725.      1708341.37       625789.76
       1707999.9       625999.75
#Sta/Elev= 30
    4809  450.17    4819  448.09    4829   446.5    4859  440.14    4869  438.74
    4899   433.4    4909  431.02    4919  428.05    4929  424.73    4939     421
    4949  417.91    4969  413.71    4979  409.77  4983.3  405.18  4984.8  402.18
  5015.2  402.18  5016.7  405.18  5043.7  410.02  5053.7   410.6  5073.7  410.68
  5083.7  411.38  5103.7  413.55  5123.7  414.51  5173.7  415.22  5243.7  418.12
  5283.7  420.17  5313.7  423.62  5323.7  425.07  5383.7  436.87  5404.6   439.7
#Mann= 3 ,-1 , 0
    4809     .15       0  4983.3     .05       0  5016.7     .13       0
Bank Sta=4983.3,5016.7
Exp/Cntr=0.3,0.1

Type RM Length L Ch R = 1 ,18000   ,500,500,500
BEGIN DESCRIPTION:
Barnes Creek 36.0
END DESCRIPTION:
XS GIS Cut Line= 3
      1708206.21       625241.98      1708063.29       625372.72
      1707841.06         625640.
#Sta/Elev= 26
  4806.3  430.64  4836.3  427.57  4886.3  424.45  4896.3  424.15  4946.3  425.61
  4956.3  424.67  4966.3  422.18  4976.3   412.8  4983.3  401.09  4984.8  398.09
  5015.2  398.09  5016.7  401.09    5030  406.24    5060  410.13    5100  412.05
    5130  411.15    5160  411.56    5180  412.58    5190  413.49    5200  414.15
    5250  416.32    5290     420    5300  421.26    5330  427.16    5340  430.06
  5347.6  432.49
#Mann= 3 ,-1 , 0
  4806.3     .15       0  4983.3     .05       0  5016.7     .13       0
Bank Sta=4983.3,5016.7
Exp/Cntr=0.3,0.1

Type RM Length L Ch R = 1 ,17500   ,473,473,473
BEGIN DESCRIPTION:
Barnes Creek 35.0
END DESCRIPTION:
XS GIS Cut Line= 3
      1708038.25       624794.58      1707741.24       624991.59
      1707552.54       625150.65
#Sta/Elev= 29
  4643.6  436.38  4683.6   430.4  4723.6  425.89  4793.6  420.02  4803.6  419.68
  4823.6  419.97  4853.6  421.88  4933.6  422.41  4973.6  420.74  4983.3  399.37
  4984.8  396.37  5015.2  396.37  5016.7  399.37    5020  410.45    5030  408.79
    5040  406.34    5050   405.4    5090  406.97    5120  409.06    5140  409.82
    5150  410.74    5160  412.01    5170  414.81    5190  421.57    5200  425.59
    5210  428.38    5220  430.53    5230  433.44  5246.8  436.51
#Mann= 3 ,-1 , 0
  4643.6     .15       0  4983.3     .05       0  5016.7     .15       0
Bank Sta=4983.3,5016.7
Exp/Cntr=0.3,0.1

Type RM Length L Ch R = 1 ,17027   ,623,623,623
BEGIN DESCRIPTION:
Barnes Creek 34.0
END DESCRIPTION:
XS GIS Cut Line= 3
      1707764.34       624498.77      1707638.35       624560.85
      1707450.29       624708.75
#Sta/Elev= 28
  4860.4  434.18  4870.4  430.94  4880.4  428.45  4900.4  425.64  4920.4  422.11
  4930.4  420.93  4940.4   420.2  4980.4   415.2  4983.3  400.27  4984.8  397.27
  5015.2  397.27  5016.7  400.27  5020.8  407.84  5030.8  407.42  5040.8  407.27
  5050.8  406.61  5060.8  405.47  5070.8  403.49  5080.8  402.27  5100.8  400.93
  5130.8  404.19  5140.8  406.18  5150.8  407.54  5160.8  410.29  5180.8  416.75
  5210.8  423.25  5220.8  424.74  5240.1  426.94
#Mann= 3 ,-1 , 0
  4860.4     .15       0  4983.3     .05       0  5016.7     .15       0
Bank Sta=4983.3,5016.7
Exp/Cntr=0.3,0.1

Type RM Length L Ch R = 1 ,16404   ,497,497,497
BEGIN DESCRIPTION:
Barnes Creek 33.0
END DESCRIPTION:
XS GIS Cut Line= 3
      1707360.79       624025.85      1707296.89       624106.18
      1707152.66       624268.66
#Sta/Elev= 18
  4898.7  429.21  4918.7  425.83  4928.7   423.4  4948.7  416.08  4958.7  411.12
  4978.7  401.72  4983.3  398.47  4984.8  395.47  5015.2  395.47  5016.7  398.47
  5021.3   399.4  5041.3  400.86  5051.3  402.49  5091.3  407.21  5111.3  408.81
  5131.3  411.41  5171.3  414.99  5218.6  417.51
#Mann= 3 ,-1 , 0
  4898.7     .15       0  4983.3     .05       0  5016.7     .15       0
Bank Sta=4983.3,5016.7
Exp/Cntr=0.3,0.1

Type RM Length L Ch R = 1 ,15907   ,503,503,503
BEGIN DESCRIPTION:
Barnes Creek 32.0
END DESCRIPTION:
XS GIS Cut Line= 3
      1707495.88       623808.51      1707285.93       623684.37
      1707220.21       623646.03
#Sta/Elev= 20
  4756.9  420.55  4766.9  419.29  4776.9  417.55  4796.9  414.97  4816.9  410.41
  4826.9  408.44  4836.9  405.79  4846.9  405.04  4896.9  405.07  4906.9   404.4
  4916.9  402.64  4926.9  401.75  4936.9  400.49  4966.9  395.52  4983.3  392.86
  4984.8  389.86  5015.2  389.86  5016.7  392.86  5060.8  417.69  5076.9  422.21
#Mann= 3 ,-1 , 0
  4756.9     .15       0  4983.3     .05       0  5016.7     .15       0
Bank Sta=4983.3,5016.7
Exp/Cntr=0.3,0.1

Type RM Length L Ch R = 1 ,15404   ,904,904,904
BEGIN DESCRIPTION:
Barnes Creek 31.0
END DESCRIPTION:
XS GIS Cut Line= 3
      1707872.08       623487.16      1707640.18       623326.47
      1707581.72       623258.88
#Sta/Elev= 26
  4716.2  423.69  4726.2  423.39  4746.2  419.14  4756.2  417.33  4766.2  415.06
  4786.2  409.71  4806.2  403.58  4816.2  401.33  4826.2  400.53  4836.2  400.12
  4856.2  400.01  4886.2  401.16  4906.2  400.48  4916.2  399.88  4926.2  398.29
  4936.2     398  4946.2  398.25  4966.2  397.43  4976.2  396.76  4983.3   392.7
  4984.8   389.7  5015.2   389.7  5016.7   392.7  5068.3  416.26  5078.3  418.74
  5087.7  420.32
#Mann= 3 ,-1 , 0
  4716.2     .15       0  4983.3     .05       0  5016.7     .15       0
Bank Sta=4983.3,5016.7
Exp/Cntr=0.3,0.1

Type RM Length L Ch R = 1 ,14500   ,755,755,755
BEGIN DESCRIPTION:
Barnes Creek 29.0
END DESCRIPTION:
XS GIS Cut Line= 3
      1708387.29       622862.89      1708299.08       622868.69
       1707700.2       623034.08
#Sta/Elev= 28
  4911.6  433.25  4921.6  433.15  4931.6  431.67  4941.6  426.84  4971.6  401.77
  4981.6  399.14    4983  389.02  4984.5  386.02  5015.5  386.02    5017  389.02
    5030  391.49    5220  397.54    5250  397.55    5290  398.98    5330  397.68
    5370  397.31    5380  395.75    5400  391.75    5410  397.64    5420   398.3
    5460   401.5    5490   402.6    5520  402.53    5540  403.28    5580  403.79
    5600  405.57    5610  406.76  5621.3  409.09
#Mann= 4 ,-1 , 0
  4911.6     .15       0    4983     .05       0    5017     .15       0
    5290      10       0
Bank Sta=4983,5017
Exp/Cntr=0.3,0.1

Type RM Length L Ch R = 1 ,13745   ,380,380,380
BEGIN DESCRIPTION:
Barnes Creek 28.0
END DESCRIPTION:
XS GIS Cut Line= 3
      1707825.74       622404.11      1707718.47        622561.6
      1707604.33       622762.49
#Sta/Elev= 27
  4799.2  413.13  4809.2  412.48  4819.2  410.77  4829.2  406.03  4839.2  400.22
  4849.2  398.24  4859.2  399.15  4869.2  400.78  4879.2  401.09  4909.2  399.71
  4919.2  398.23  4929.2  397.05  4939.2  395.57  4969.2   388.9  4979.2   387.6
    4983  385.08  4984.5  382.08  5015.5  382.08    5017  385.08  5029.8  389.89
  5109.8   393.8  5129.8  395.02  5159.8  399.29  5179.8  402.91  5209.8  411.62
  5219.8  413.85  5220.8     414
#Mann= 3 ,-1 , 0
  4799.2     .15       0    4983     .05       0    5017     .15       0
Bank Sta=4983,5017
Exp/Cntr=0.3,0.1

Type RM Length L Ch R = 1 ,13365   ,427,427,427
BEGIN DESCRIPTION:
Barnes Creek 27.0
END DESCRIPTION:
XS GIS Cut Line= 3
       1707506.2       622184.95      1707476.52       622315.09
      1707449.13       622495.44
#Sta/Elev= 14
  4865.8  402.66  4875.8  400.27    4983   380.9  4984.5   377.9  5015.5   377.9
    5017   380.9  5049.3  387.82  5059.3  389.77  5069.3  392.57  5079.3  395.66
  5089.3  398.28  5099.3  399.67  5119.3  400.51  5181.7  405.65
#Mann= 3 ,-1 , 0
  4865.8     .15       0    4983     .05       0    5017     .15       0
Bank Sta=4983,5017
Exp/Cntr=0.3,0.1

Type RM Length L Ch R = 1 ,12938   ,755,755,755
BEGIN DESCRIPTION:
Barnes Creek 26.0
END DESCRIPTION:
XS GIS Cut Line= 3
      1707061.11       622095.98      1707051.98       622299.11
      1707061.11       622493.16
#Sta/Elev= 26
  4793.9  414.87  4803.9  411.19  4823.9  402.51  4833.9  398.47  4843.9   394.8
  4853.9   391.9  4863.9  389.94  4873.9  388.69  4923.9  385.12  4953.9  381.12
    4983  378.15  4984.5  375.15  5015.5  375.15    5017  378.15  5017.2  383.45
  5067.2  387.95  5077.2  388.15  5087.2   388.1  5097.2  388.93  5117.2   389.9
  5137.2  391.48  5147.2  393.36  5167.2  399.02  5177.2  402.31  5187.2  406.15
  5191.5  407.98
#Mann= 3 ,-1 , 0
  4793.9     .15       0    4983     .05       0    5017     .15       0
Bank Sta=4983,5017
Exp/Cntr=0.3,0.1

Type RM Length L Ch R = 1 ,12183   ,494,494,494
BEGIN DESCRIPTION:
Barnes Creek 25.0
END DESCRIPTION:
XS GIS Cut Line= 3
      1706561.27       621915.62      1706319.29       622171.29
      1706232.57       622326.48
#Sta/Elev= 30
  4647.1  408.79  4657.1  405.95  4687.1  398.26  4717.1  391.38  4727.1  389.82
  4807.1  384.13  4817.1  384.15  4837.1  383.53  4867.1  383.64  4917.1  380.28
  4937.1   379.8  4967.1  377.57  4977.1  376.52    4983  374.92  4984.5  371.92
  5015.5  371.92    5017  374.92  5019.1   376.8  5039.1  378.02  5049.1  380.28
  5059.1  381.39  5069.1  382.97  5079.1  385.27  5099.1  387.27  5109.1  388.61
  5119.1  390.45  5139.1  397.66  5159.1  406.92  5169.1  410.97  5176.9  413.68
#Mann= 3 ,-1 , 0
  4647.1     .15       0    4983     .05       0    5017     .15       0
Bank Sta=4983,5017
Exp/Cntr=0.3,0.1

Type RM Length L Ch R = 1 ,11689   ,689,689,689
BEGIN DESCRIPTION:
Barnes Creek 24.0
END DESCRIPTION:
XS GIS Cut Line= 3
      1706490.43       621780.99      1705958.65       621849.46
      1705803.49       621867.71
#Sta/Elev= 27
    4465  406.76    4475   404.9    4485  402.79    4525   391.6    4535   389.8
    4545  388.72    4605  384.87    4735  381.84    4785  381.83    4805  382.14
    4855  381.43    4885  379.72    4955  377.53    4965  376.96    4975  375.13
    4983  372.39  4984.5  369.39  5015.5  369.39    5017  372.39  5031.2  372.95
  5041.2  373.71  5091.2  384.71  5111.2  388.35  5131.2  394.66  5141.2  399.03
  5151.2  403.94  5157.4  407.38
#Mann= 3 ,-1 , 0
    4465     .15       0    4983     .05       0    5017     .15       0
Bank Sta=4983,5017
Exp/Cntr=0.3,0.1

Type RM Length L Ch R = 1 ,11000   ,500,500,500
BEGIN DESCRIPTION:
Barnes Creek 22.0
END DESCRIPTION:
XS GIS Cut Line= 3
      1706239.44       621166.99      1705972.25       621169.99
      1705750.92        621164.7
#Sta/Elev= 30
  4732.8  404.13  4742.8  400.52  4782.8   387.8  4802.8  380.46  4812.8  379.16
  4832.8   377.7  4882.8  376.84  4902.8  377.33  4922.8  376.87  4932.8  376.35
  4962.8  373.49  4972.8  371.85  4982.8  369.95    4983  366.23  4984.5  363.23
  5015.5  363.23    5017  366.23    5020  367.55    5030  371.43    5040  373.52
    5070  374.54    5120  377.55    5150  379.99    5160   381.1    5170  382.72
    5190  386.96    5200  390.64    5210  394.74    5220  399.32  5221.4   400.1
#Mann= 3 ,-1 , 0
  4732.8     .15       0    4983     .05       0    5017     .15       0
Bank Sta=4983,5017
Exp/Cntr=0.3,0.1

Type RM Length L Ch R = 1 ,10500   ,500,500,500
BEGIN DESCRIPTION:
Barnes Creek 21.0
END DESCRIPTION:
XS GIS Cut Line= 3
       1706392.3       620776.67      1706035.37       620678.81
      1705734.96       620614.62
#Sta/Elev= 30
  4629.9  396.94  4679.9  388.22  4709.9  384.26  4779.9  376.44  4789.9  375.93
  4799.9  376.06  4829.9  374.64  4859.9  374.18  4889.9  374.93  4919.9  374.95
  4929.9  374.59  4939.9  373.04  4949.9  372.53  4979.9  372.05    4983  365.81
  4984.5  362.81  5015.5  362.81    5017  365.81    5020  372.33    5030  372.52
    5050  374.07    5090  374.29    5170  376.96    5210  380.85    5220  382.91
    5230  385.76    5240  388.09    5250  389.55    5300  399.85  5307.2  402.23
#Mann= 3 ,-1 , 0
  4629.9     .15       0    4983    .045       0    5017     .15       0
Bank Sta=4983,5017
Exp/Cntr=0.3,0.1

Type RM Length L Ch R = 1 ,10000   ,708,708,708
BEGIN DESCRIPTION:
Barnes Creek 20.0
END DESCRIPTION:
XS GIS Cut Line= 3
      1706538.37       620393.19      1706247.91       620233.63
      1705849.13       620046.29
#Sta/Elev= 30
  4668.6  401.93  4678.6  397.96  4708.6  384.66  4748.6  370.05  4768.6  371.67
  4808.6  370.71  4838.6  371.16  4858.6   372.1  4898.6  371.94  4918.6  372.94
  4938.6  372.64  4948.6  372.22  4958.6   370.1  4968.6  366.51    4983  365.15
  4984.5  362.15  5015.5  362.15    5017  365.15    5020  369.96    5030  371.38
    5120  372.25    5170  371.49    5190  370.63    5210  371.13    5230   370.5
    5270  371.55    5280  371.35    5320  375.92    5430  391.02  5440.6  391.32
#Mann= 3 ,-1 , 0
  4668.6     .15       0    4983    .045       0    5017     .15       0
Bank Sta=4983,5017
Exp/Cntr=0.3,0.1

Type RM Length L Ch R = 1 ,9292    ,430,430,430
BEGIN DESCRIPTION:
Barnes Creek 19.0
END DESCRIPTION:
XS GIS Cut Line= 3
      1706294.21       619308.99      1705860.51       619838.57
      1705766.93        619925.3
#Sta/Elev= 30
  4316.8  399.53  4336.8  392.16  4366.8  379.19  4376.8  374.24  4386.8  370.11
  4396.8   368.7  4406.8  368.28  4486.8   367.5  4496.8  367.05  4506.8  365.85
  4516.8   365.7  4536.8  366.47  4556.8  366.16  4656.8  367.21  4676.8  368.28
  4746.8  368.37  4786.8  368.79  4806.8  368.27  4826.8  368.55  4846.8  368.03
  4896.8  368.05  4956.8  366.14  4976.8  364.78    4982  361.46  4983.5  358.46
  5016.5  358.46    5018  361.46  5041.3  370.73  5091.3  381.74  5128.9   388.2
#Mann= 3 ,-1 , 0
  4316.8     .15       0    4982    .045       0    5018     .15       0
Bank Sta=4982,5018
Exp/Cntr=0.3,0.1

Type RM Length L Ch R = 1 ,8862    ,442,442,442
BEGIN DESCRIPTION:
Barnes Creek 18.0
END DESCRIPTION:
XS GIS Cut Line= 3
      1705566.07       619466.49      1705524.98       619587.49
      1705463.35        619806.6
#Sta/Elev= 18
    4874  387.21    4914  375.22    4934   367.2    4944  364.23    4954  363.18
    4964   361.7    4974  359.87    4982  356.27  4983.5  353.27  5016.5  353.27
    5018  356.27  5061.8  362.56  5081.8  363.04  5101.8  364.68  5121.8  365.56
  5211.8  373.36  5221.8  375.31  5229.4  378.94
#Mann= 3 ,-1 , 0
    4874     .15       0    4982    .045       0    5018     .15       0
Bank Sta=4982,5018
Exp/Cntr=0.3,0.1
